HEC-RAS study AshepooRiver.prj: S-15-41 over Ashepoo River

--- AshepooRiver.g03 (geometry) --- (continued)

Type RM Length L Ch R = 1 ,57186   ,742.9,742.9,742.9
BEGIN DESCRIPTION:
HEC-2 RS: 216847
END DESCRIPTION:
XS GIS Cut Line= 6
2113486.58521938345768.4686934842113057.02499013344616.224982676
2112606.63455243343774.9088022842112213.00337047343643.294728209
2109864.08764517343298.3666103682107113.53128844343196.340419961
#Sta/Elev= 30
       0   22.14   160.9   22.19   401.6   17.03   774.8   16.64   894.7   12.41
   915.5    9.28     979    7.29  1172.3    5.43    1193    7.43  1584.5    8.22
  1599.4    6.41    1621    9.12  1636.7     7.6  1886.1    6.59  2083.4    6.31
  2099.5    8.28  2150.4     6.5  2360.7    7.45  2384.9    3.86    2700    3.69
 2737.58   -2.36 2846.02   -2.34 2881.093.846987  3067.5    3.81    3379    8.01
  4976.3    6.31  6136.1   11.42  7219.6   11.57  7577.5   12.93    7729   16.28
#Mann= 3 ,-1,0
       0     .12       0    2700    .041       0 2881.09     .12       0
Bank Sta=2700,2881.09
XS Rating Curve= 0 ,0
Exp/Cntr(USF)=0,0
Exp/Cntr=0.3,0.1

Type RM Length L Ch R = 1 ,56443   ,980.8,980.8,980.8
BEGIN DESCRIPTION:
HEC-2 RS: 215997
END DESCRIPTION:
XS GIS Cut Line= 6
 2113542.7384924345627.2632154992112982.60128618343689.622050567
2112594.04871233342810.1317107832111140.64623269343026.164538765
2109541.92443561342933.8618398392107232.32289834342975.171662578
#Sta/Elev= 30
       0   22.56   351.7   19.48   589.4   19.52   783.5    13.7   800.5    8.91
   831.1    7.36     855    8.89   878.8    6.89  1072.8    5.49  1552.4    8.84
  1583.5    6.74  1603.9    9.51  1665.2    7.52  2467.9    5.74  2955.8    7.57
  3078.6    7.19  3222.5     3.5    3620 3.73413 3669.99   -2.64 3829.28   -2.65
 3846.123.762544  4003.1    3.94  4115.4    8.47    4998     8.3  5662.3       6
  6588.3   10.69  7330.1   10.86  7563.1   13.41  8144.1   12.84  8363.9   15.81
#Mann= 3 ,-1,0
       0     .12       0    3620    .041       0 3846.12     .12       0
Bank Sta=3620,3846.12
XS Rating Curve= 0 ,0
Exp/Cntr(USF)=0,0
Exp/Cntr=0.3,0.1

Type RM Length L Ch R = 1 ,55462   ,1590.3,1590.3,1590.3
BEGIN DESCRIPTION:
HEC-2 RS: 215090 (LTR M)
END DESCRIPTION:
Node Name=M
XS GIS Cut Line= 6
2113568.81423419345468.007339637 2112947.9376938342607.997925717
2112732.08088266342287.2343462792112321.38115258342037.902023321
2109072.61770797342788.5819753352107403.45554704  342823.5553852
#Sta/Elev= 30
       0   20.41   536.7   19.98   566.8   12.46   640.4    7.62   683.9    10.8
   744.1    7.28   954.8    5.69    1224    8.51  1526.9    6.69  1543.5    9.19
  2068.7    6.78  3053.7    7.79    3180     8.6  3215.6   11.06  3230.4    9.11
  3530.1    7.26  4254.4    7.53  4425.2    3.75    46253.314335 4644.54    -2.9
 4768.05   -2.88 4790.713.322143    5492     5.1  5714.1    8.53  6326.5    5.43
  6676.4    9.23  7916.8   10.41  8360.3   14.39  8629.8   12.83  8803.3   14.52
#Mann= 3 ,-1,0
       0     .12       0    4625    .041       0 4790.71     .12       0
Bank Sta=4625,4790.71
XS Rating Curve= 0 ,0
Exp/Cntr(USF)=0,0
Exp/Cntr=0.3,0.1

Type RM Length L Ch R = 1 ,53872   ,1068.4,1068.4,1068.4
BEGIN DESCRIPTION:
HEC-2 RS: 214067
END DESCRIPTION:
XS GIS Cut Line= 6
2113665.95705568 345426.336509692113086.88115373342163.439416852
2112369.53776723341723.0682256752111241.00129154341342.111761542
2109965.28864871341437.8266651632107086.50153097342275.881131254
#Sta/Elev= 30
       0    20.4   338.9   21.36   379.5   24.94     503   12.22   549.7   13.56
   713.2    7.74   773.5    9.25   960.1    6.18  1661.4    8.73  3006.1    7.73
  3073.2    9.67  4510.9    7.78  5103.9   12.69  5380.9    9.59    5404    4.56
  5661.7     4.2  5687.9    7.93    5708    4.63  5840.1    3.24    61103.904998
 6125.35    -3.5 6246.04   -3.48 6282.263.966102  7423.3    5.85  7582.9    9.89
  7891.5   11.31  8155.4    8.09  8513.9    8.19    8889   10.35  9654.2   21.11
#Mann= 3 ,-1,0
       0     .12       0    6110    .041       0 6282.26     .12       0
#XS Ineff= 1 ,-1
 7904.23 8907.04   11.37
Permanent Ineff=
       T
Bank Sta=6110,6282.26
XS Rating Curve= 0 ,0
Exp/Cntr(USF)=0,0
Exp/Cntr=0.3,0.1

Type RM Length L Ch R = 1 ,52803   ,839.1,839.1,839.1
BEGIN DESCRIPTION:
HEC-2 RS: 213236
END DESCRIPTION:
XS GIS Cut Line= 6
2113710.59355572345430.4006670612113448.33330875343148.228105745
2113086.53357444341637.1573886812112748.97970278 341217.20142283
2110755.64770619340490.302856961 2109124.3484468339515.562594273
#Sta/Elev= 30
       0   21.75    23.1   22.74    66.1   20.11   272.6   23.09   416.2   22.35
   630.7   14.05   667.3   14.56   743.3     8.1  1004.2    6.41  1859.8    8.46
  2984.3    7.55  3436.5   10.03    4285     7.1  4990.1    8.73  5396.3   13.23
  5722.9    9.98  5840.9    6.54  6413.2    8.12    66603.492058 6676.48   -3.69
 6760.69   -3.67 6780.463.485386  7219.8    3.44    7428   16.88  7618.6   19.79
  8120.2   17.53  8202.9    19.2  8237.4   16.87  8252.8   19.51  8415.8   18.21
#Mann= 3 ,-1,0
       0     .12       0    6660    .041       0 6780.46     .12       0
Bank Sta=6660,6780.46
XS Rating Curve= 0 ,0
Exp/Cntr(USF)=0,0
Exp/Cntr=0.3,0.1

Type RM Length L Ch R = 1 ,51964   ,952,952,952
BEGIN DESCRIPTION:
HEC-2 RS: 212304
END DESCRIPTION:
XS GIS Cut Line= 6
2113753.67471267345423.5593204752113580.43345627 343190.64241309
2113183.51759426340879.1236672472111775.48857235340489.480415901
2111290.56987558 339988.659403132110252.98432053338783.358492686
#Sta/Elev= 30
       0   22.82   500.9   21.65   787.2    8.57  1027.4     6.3  2900.5    7.38
  2960.4    9.76  3108.2    7.37    3433   10.97  4048.6    5.98  4603.5    7.27
  4627.1   11.74  4647.4    6.79  5381.2    7.66  5401.5   11.21  5431.7    7.79
  5585.5   11.34  5854.9    8.51  6167.8    11.2  6548.8    2.84    6710 3.13754
 6716.82   -4.04 6786.62   -4.04 6797.952.897896  7392.1    3.16  7509.4    9.29
  7782.9   15.57  8117.3   15.28  8171.1   13.07  8189.7    15.2  8336.2   14.65
#Mann= 3 ,-1,0
       0     .12       0    6710    .041       0 6797.95     .12       0
Bank Sta=6710,6797.95
XS Rating Curve= 0 ,0
Exp/Cntr(USF)=0,0
Exp/Cntr=0.3,0.1

Type RM Length L Ch R = 1 ,51012   ,948.3,948.3,948.3
BEGIN DESCRIPTION:
HEC-2 RS: 211308
END DESCRIPTION:
XS GIS Cut Line= 6
2113784.01759306345418.4051467052113720.27176802342893.723116748
2113327.76276237340738.0580405182112459.28196653340443.410629815
2111632.31338533338680.5684926832111419.26402097337778.426294558
#Sta/Elev= 30
       0   24.26   491.3    21.5   836.3    8.39  1072.6    6.43  2267.3    8.96
  3265.6    7.35  3552.6    9.96  4400.8     5.8  4843.4    7.49  4863.7   11.17
  4887.2    6.78  5462.6    6.96  5562.3    7.49  5583.7   11.67  5601.8     7.7
  5640.9    9.71  6244.7    9.99  6268.6    5.74  6291.6    8.56    6456    2.64
    68003.201209 6808.59   -4.28 6905.56   -4.28 6924.723.132063  7367.3    2.75
  7500.2    8.17  7828.2   11.04  8087.9    9.79  8263.2   16.23  8555.3   17.53
#Mann= 3 ,-1,0
       0     .12       0    6800    .041       0 6924.72     .12       0
Bank Sta=6800,6924.72
XS Rating Curve= 0 ,0
Exp/Cntr(USF)=0,0
Exp/Cntr=0.3,0.1

Type RM Length L Ch R = 1 ,50064   ,797,797,797
BEGIN DESCRIPTION:
HEC-2 RS: 210260
END DESCRIPTION:
XS GIS Cut Line= 6
2113819.67999959345380.3975931412113927.97080106342095.905734601
2113711.50232809341102.1186541492113127.51502048340019.569395021
2112880.30446054339219.3152655542112811.38049324338267.623629299
#Sta/Elev= 30
       0   25.31   439.5   21.89   888.8    7.93    1030    6.85  1049.7    8.48
  1069.4    6.29  1401.1    8.26  2431.8    7.18  2484.6    9.58    2501    7.33
  2602.9    6.95  3336.4    8.99    3602    7.66  3678.4    9.03  3701.6    7.37
  3818.2    9.21  3961.6    6.43  4659.4    5.41    4979    8.44  5351.9    8.86
  5482.1    7.73  5650.7    2.32    64603.021096 6470.79   -4.76 6557.69    -4.8
 6585.91    2.83  6631.7     9.9  6694.2   13.81  7180.9   24.77  7330.7   25.16
#Mann= 3 ,-1,0
       0     .12       0    6460    .041       0 6585.91     .12       0
Bank Sta=6460,6585.91
XS Rating Curve= 0 ,0
Exp/Cntr(USF)=0,0
Exp/Cntr=0.3,0.1

Type RM Length L Ch R = 1 ,49267   ,1164.1,1164.1,1164.1
BEGIN DESCRIPTION:
HEC-2 RS: 209434
END DESCRIPTION:
XS GIS Cut Line= 6
2113842.64379361  345402.5263264 2114026.3655615343394.716572421
2114248.95082345341596.1784298422114134.59979798341062.760749973
2113770.53918435 340068.973669522113505.26959665337962.936515315
#Sta/Elev= 30
       0   24.54   456.4   22.61   634.4   18.91   861.8   10.76  1033.3    7.32
  1125.4    7.86  1145.2    6.16  1395.7    8.16  2336.8    8.51  2858.5    6.84
  3007.3    8.59  3060.2    7.06    3424    7.13    3705   10.32  4923.2    4.84
  5342.6    8.88  5499.5    8.37  5582.1    2.62  5651.4    1.79  5687.8    3.17
    64002.261818 6414.62   -5.28 6463.46   -5.25 6477.612.433743  6507.1    2.75
  6546.8    11.2  6639.6   17.08  6958.3   28.45  7119.9    25.7  7555.2   25.48
#Mann= 3 ,-1,0
       0     .12       0    6400    .041       0 6477.61     .12       0
Bank Sta=6400,6477.61
XS Rating Curve= 0 ,0
Exp/Cntr(USF)=0,0
Exp/Cntr=0.3,0.1

Type RM Length L Ch R = 1 ,48103   ,717.4,717.4,717.4
BEGIN DESCRIPTION:
HEC-2 RS: 208274 (LTR L)
END DESCRIPTION:
Node Name=L
XS GIS Cut Line= 6
2113877.86478229345392.9455559052113984.30492154344357.593753259
2114390.07680005 341709.099288592114726.00750383339431.354087047
 2114725.9193221338789.0864046892114276.75018094338049.327786138
#Sta/Elev= 30
       0   24.48   216.4    22.3   328.5   23.53   516.6   22.26   589.2   16.95
   661.7   18.21   780.5    12.9   981.8    7.41  1160.7    6.32  1177.3    8.38
  1200.5    7.07  1635.5    8.26  1974.1    6.62    3342    6.86  3521.3    8.31
  3553.3   10.56  3564.4    8.91  3769.4   10.45  5223.3    4.81  5346.1    2.86
 5947.11    2.21  5972.7   -5.57 6051.68   -5.57 6069.96    2.31  6331.3    1.84
  6518.3   10.25  6789.1   15.57  6939.3   11.69  7073.2      16  7530.4   22.27
#Mann= 3 ,-1,0
       0     .12       0 5947.11    .041       0 6069.96     .12       0
Bank Sta=5947.11,6069.96
XS Rating Curve= 0 ,0
Exp/Cntr(USF)=0,0
Exp/Cntr=0.5,0.3

Type RM Length L Ch R = 1 ,47386   ,148.2,148.2,148.2
BEGIN DESCRIPTION:
HEC-2 RS: 207385
END DESCRIPTION:
XS GIS Cut Line= 5
2113961.77074045345415.0293650792114204.83077183344471.731700322
2115437.79764054339477.5591892312115543.63379055339062.969763302
2116067.18892544336966.980577882
#Sta/Elev= 30
       0   21.12   631.4    19.6   885.6   12.16  1227.2    6.59  1930.4    7.99
  2863.3     5.9  2971.5     7.5  3208.1    5.84  3285.9    7.39  3738.9    6.93
    3962   10.31  4523.1    7.35  4969.3    7.52  5374.9    2.87  6021.8    1.63
 6040.13   -5.91 6149.65   -5.91 6171.84    1.71  6579.2    2.12  6704.4    4.32
  6717.9    2.45  6755.2    4.94  6856.6     2.6  6978.4     3.1  7232.1    7.42
  7879.2   12.37  8334.8   11.55    8416    9.54  8473.5   13.37  8706.5   12.71
#Mann= 3 ,-1,0
       0     .12       0  6021.8    .041       0 6171.84     .12       0
#XS Ineff= 2 , 0
            5955   10.27    6215            9.53
Permanent Ineff=
       F       F
Bank Sta=6021.8,6171.84
XS Rating Curve= 0 ,0
Exp/Cntr(USF)=0,0
Exp/Cntr=0.5,0.3

Type RM Length L Ch R = 3 ,47296   ,,,
BEGIN DESCRIPTION:
SC-303 over Ashepoo River
END DESCRIPTION:
Bridge Culvert--1,0,-1,-1, 0
Deck Dist Width WeirC Skew NumUp NumDn MinLoCord MaxHiCord MaxSubmerge Is_Ogee
25,90,2.6,0, 14, 14, , , 0.98, 0, 2,2,,
       0    1000 5979.99    5980    5980    6190    6190 6190.01    6300    6600
    7000    7200    8000    8800
  20.657  14.031   10.26   10.26   10.26   10.22   10.22   10.22     9.9     9.7
    9.53   9.531   13.56   15.26
                                    8.57    8.53
                                
       0    1000 5979.99    5980    5980    6190    6190 6190.01    6300    6900
    7000    7200    8000    8800
  20.657  14.031   10.26   10.26   10.26   10.22   10.22   10.22     9.9     9.7
    9.53   9.531   13.56   15.26
                                    8.57    8.53
                                
Pier Skew, UpSta & Num, DnSta & Num=  ,5995, 2 ,5995, 2 , 0 , 0 , 0 ,,
     1.5     1.5
      -6    9.95
     1.5     1.5
      -6    9.95
Pier Skew, UpSta & Num, DnSta & Num=  ,6010, 2 ,6010, 2 , 0 , 0 , 0 ,,
     1.5     1.5
   -5.91    9.95
     1.5     1.5
   -5.91    9.95
Pier Skew, UpSta & Num, DnSta & Num=  ,6025, 2 ,6025, 2 , 0 , 0 , 0 ,,
     1.5     1.5
      -6    9.95
     1.5     1.5
      -6    9.95
Pier Skew, UpSta & Num, DnSta & Num=  ,6040, 2 ,6040, 2 , 0 , 0 , 0 ,,
     1.5     1.5
   -5.91    9.95
     1.5     1.5
   -5.91    9.95
Pier Skew, UpSta & Num, DnSta & Num=  ,6055, 2 ,6055, 2 , 0 , 0 , 0 ,,
     1.5     1.5
      -6    9.95
     1.5     1.5
      -6    9.95
Pier Skew, UpSta & Num, DnSta & Num=  ,6070, 2 ,6070, 2 , 0 , 0 , 0 ,,
     1.5     1.5
   -5.91    9.95
     1.5     1.5
   -5.91    9.95
Pier Skew, UpSta & Num, DnSta & Num=  ,6085, 2 ,6085, 2 , 0 , 0 , 0 ,,
     1.5     1.5
      -6    9.95
     1.5     1.5
      -6    9.95
Pier Skew, UpSta & Num, DnSta & Num=  ,6100, 2 ,6100, 2 , 0 , 0 , 0 ,,
     1.5     1.5
   -5.91    9.95
     1.5     1.5
   -5.91    9.95
Pier Skew, UpSta & Num, DnSta & Num=  ,6115, 2 ,6115, 2 , 0 , 0 , 0 ,,
     1.5     1.5
      -6    9.95
     1.5     1.5
      -6    9.95
Pier Skew, UpSta & Num, DnSta & Num=  ,6130, 2 ,6130, 2 , 0 , 0 , 0 ,,
     1.5     1.5
   -5.91    9.95
     1.5     1.5
   -5.91    9.95
Pier Skew, UpSta & Num, DnSta & Num=  ,6145, 2 ,6145, 2 , 0 , 0 , 0 ,,
     1.5     1.5
      -6    9.95
     1.5     1.5
      -6    9.95
Pier Skew, UpSta & Num, DnSta & Num=  ,6160, 2 ,6160, 2 , 0 , 0 , 0 ,,
     1.5     1.5
   -5.91    9.95
     1.5     1.5
   -5.91    9.95
Pier Skew, UpSta & Num, DnSta & Num=  ,6175, 2 ,6175, 2 , 0 , 0 , 0 ,,
     1.5     1.5
      -6    9.95
     1.5     1.5
      -6    9.95
Abutment Skew #Up #Dn= , 3 , 3
    5980    5982  5990.7
    6.57    6.57    2.22
    5980    5982  5990.7
    6.57    6.57    2.22
Abutment Skew #Up #Dn= , 3 , 3
 6178.38    6188    6190
    1.72    6.53    6.53
 6178.38    6188    6190
    1.72    6.53    6.53
BR Coef=-1 ,-1 ,-1 ,0.9, 0 ,,,0.8,0,1.2,0,
WSPro=,,,, 1 ,,,, 0 ,,,, 0 ,,,,-1 ,-1 ,-1 , 0 , 0 , 0 , 0 , 0
BC Design=,, 0 ,, 0 ,,,,,,
BC Use User HTab Curves=0
BC User HTab FreeFlow(D)= 0

Type RM Length L Ch R = 1 ,47238   ,831.2,831.2,831.2
BEGIN DESCRIPTION:
HEC-2 RS: 207243
END DESCRIPTION:
XS GIS Cut Line= 6
2114073.47904332  345423.60386612114221.42584184344858.595689091
2114341.76739176344471.5221031752115658.66614636339198.105657315
2116169.30860132337126.505086102 2116213.6270204336961.916215067
#Sta/Elev= 30
       0   19.02   264.9   17.61     292   22.29   511.5   18.54     611   20.12
   784.4    12.4   860.3   16.11  1032.8    8.78  1455.5    6.82  3094.8    5.78
  4099.9    9.86  4394.1    6.23  4580.1    8.19  4901.3    7.19  4946.1    4.58
    60201.697643 6035.72   -4.72 6157.21   -4.73  6170.8    1.84  6451.8    2.25
  6518.1    5.82  6735.6    3.62  6769.4    7.54  6789.7    7.04  6803.2    3.56
  7107.5    8.56  7202.2    6.31  8216.2   15.36  8533.9   13.35  8728.9   16.04
#Mann= 3 ,-1,0
       0     .12       0    6020    .041       0  6170.8     .12       0
#XS Ineff= 2 , 0
            5963   10.27    6207            9.53
Permanent Ineff=
       F       F
Bank Sta=6020,6170.8
XS Rating Curve= 0 ,0
Exp/Cntr(USF)=0,0
Exp/Cntr=0.5,0.3

Type RM Length L Ch R = 1 ,46407   ,3831.1,3831.1,3831.1
BEGIN DESCRIPTION:
HEC-2 RS: 206515 (LTR K)
END DESCRIPTION:
Node Name=K
XS GIS Cut Line= 5
2115537.78628686345276.3727564262115691.65318385344076.177599645
2116229.20633682340420.1299743212116525.06356667338740.926794892
2116681.20054587337905.065912506
#Sta/Elev= 30
       0   33.03   602.4   21.07   949.8   17.58    1039    12.2    1145    9.85
  1576.1    5.82  2677.4    5.12  3453.6    9.18  3526.5    7.97  3662.5    9.05
  3728.9   12.12  3765.6   10.41  4269.6   10.98  4850.1    8.47  5233.7    1.47
 5885.54       2 5899.47   -4.92 5938.86   -4.87 5948.39     2.3  6206.1    8.96
  6316.1   10.18    6396    8.82  6419.4   10.56  6442.7    9.14  6462.7   10.98
  7006.6    20.8  7086.7   20.43  7116.8   18.25  7142.3   19.78  7460.8   18.38
#Mann= 3 ,-1,0
       0     .12       0 5885.54    .041       0 5948.39     .12       0
Bank Sta=5885.54,5948.39
XS Rating Curve= 0 ,0
Exp/Cntr(USF)=0,0
Exp/Cntr=0.3,0.1

Type RM Length L Ch R = 1 ,42576   ,5565.5,5565.5,5565.5
XS GIS Cut Line= 4
2118303.66927878346002.5906400612119278.61713182341189.752825883
2119603.39438416339740.9089025852119883.18310562338475.198019788
#Sta/Elev= 30
       0   16.75    17.9   18.69   128.4   17.57   145.1   19.33   205.4   17.25
   727.8   15.13   780.6   12.51  1404.2   13.66  1621.8   12.18  1819.4    6.39
    2325    3.45  2909.1     3.3  2927.7    5.16  2954.5    3.05  3088.5    4.53
    3199    2.47    49451.571982 4956.82   -6.77 4991.02   -6.77    50101.527162
  5175.7    1.89  5269.9    7.51  5340.5    8.16  6527.7     1.9  6813.4    3.04
  7179.7   10.18  7311.4   10.73  7482.2   14.63  7572.9   19.217691.659   20.19
#Mann= 3 ,0,0
       0     .12       0    4945    .041       0    5010     .12       0
Bank Sta=4945,5010
XS Rating Curve= 0 ,0
Exp/Cntr(USF)=0,0
Exp/Cntr=0.3,0.1

Type RM Length L Ch R = 1 ,37010   ,3738.7,3738.7,3738.7
BEGIN DESCRIPTION:
HEC-2 RS: 197805 (LTR I)
END DESCRIPTION:
Node Name=I
XS GIS Cut Line= 6
2124552.79285475345492.2516775562123836.54206595342602.273698308
2123387.02818671340830.4235865182123242.98947943340525.936698981
2123166.86284749339519.7699893162123290.64051106338653.450830175
#Sta/Elev= 30
       0   11.81   567.5   10.12  1247.1    4.54  1297.8    2.05  1324.9    6.16
  1342.8    4.29  1531.1    5.72  1980.8   12.41  1990.9   12.16  2003.9    8.61
  2014.6    10.9  2058.1   11.22  2166.8    8.58  2376.4    9.25    2985    3.03
  3506.4     3.2  3536.9    1.34  3740.9     3.2  4773.3   1.871 4798.42  -10.37
 4844.01  -10.34  4857.7   1.801  5697.1    1.79    5832    5.55  6088.7    6.14
  6247.4   13.57    6380   22.99  6433.1   24.45    6811   24.78  7026.5   22.56
#Mann= 3 ,-1,0
       0     .12       0  4773.3    .041       0  4857.7     .12       0
#XS Ineff= 1 ,-1
  243.38 1870.42    11.8
Permanent Ineff=
       T
Bank Sta=4773.3,4857.7
XS Rating Curve= 0 ,0
Exp/Cntr(USF)=0,0
Exp/Cntr=0.3,0.1

Type RM Length L Ch R = 1 ,33271   ,4264.8,4264.8,4264.8
XS GIS Cut Line= 6
2127732.46096736344794.0527805662126399.23665777 340633.47969719
2126231.03891756340225.1461509062126201.34741081340158.829709078
2126135.02888988 340045.470241962125616.70249457338667.560752107
#Sta/Elev= 30
       0   12.29   686.1    8.12  1037.6    8.16  1051.4    6.87  1075.5    8.32
  1509.8    7.84  1706.2    9.62  1723.4    7.49  1757.9    7.97  1768.2    9.64
  1971.6    8.19  2171.4    8.96  2200.2    7.35  2854.4    7.59  3649.9    1.95
    48101.658942 4847.36  -10.05 4943.36  -10.05 4964.96    1.76  5039.7    1.94
  5050.3     3.6  5106.3    2.09  5190.5    3.28    6032    2.25  6154.7    8.01
  6189.8   11.52  6224.8   18.09  6252.9   20.84  6358.1   24.27  6486.8   24.45
#Mann= 3 ,0,0
       0     .12       0    4810    .041       0 4964.96     .12       0
Bank Sta=4810,4964.96
XS Rating Curve= 0 ,0
Exp/Cntr(USF)=0,0
Exp/Cntr=0.3,0.1

Type RM Length L Ch R = 1 ,29006   ,6216.7,6216.7,6216.7
XS GIS Cut Line= 4
2130868.70562372343778.9454059382129851.97429128339809.514861452
2129448.06732359339029.5565790262128626.32556175337232.866964154
#Sta/Elev= 30
       0   11.22   941.1    7.34  2170.8    7.99    2513    6.71  2529.9    7.78
  2546.9    6.43  3217.7    1.78  3451.4    1.98  3478.5    3.31    3509       2
  3600.5    2.28  3654.7    4.24  3668.2     2.5  3688.6    3.77  3825.4    2.61
  3871.5    3.95  3932.5    2.25  4179.6     2.6    42201.439775 4245.38   -9.49
  4337.1   -9.43    43801.616352  4434.9    2.69  5425.6    1.98  5545.3    3.32
  5560.2    2.13  5703.5    1.88  5759.8    5.63    6107   13.966951.603   14.82
#Mann= 3 ,0,0
       0     .12       0    4220    .041       0    4380     .12       0
Bank Sta=4220,4380
XS Rating Curve= 0 ,0
Exp/Cntr(USF)=0,0
Exp/Cntr=0.3,0.1

Type RM Length L Ch R = 1 ,22789   ,4683.6,4683.6,4683.6
XS GIS Cut Line= 6
2132490.72681081342747.7794307372134387.27894148337969.420724765
2134045.07224507337683.6217255622133781.83632475337483.061024367
2133155.08413351337119.544753451 2131625.8087869336003.925853054
#Sta/Elev= 30
       0    9.22  2233.2    2.14  3250.1    1.09  3518.5    4.28  3553.8    1.69
  4097.5    1.62  4143.4    4.04  4182.3    1.87  4203.4    5.81  4514.2    4.63
  4574.2     1.9  4973.2    3.79  5001.4     .91  6105.7    2.62  6225.1    2.27
 6241.25   -1.71 6268.35   -11.5 6365.92   -11.5 6390.31   -1.71  6399.6    1.88
  6593.1    2.16  6638.6    5.34  6662.7     .77  6707.4     .39  7524.4      .6
  7544.2    3.49  7561.9     .49  7820.3     .63  8142.1    8.51  8535.3    13.2
#Mann= 3 ,0,0
       0     .12       0 6241.25    .041       0 6390.31     .12       0
#XS Ineff= 2 ,-1
 4985.92 5740.85    3.05 6653.52    8000    5.52
Permanent Ineff=
       T       T
Bank Sta=6241.25,6390.31
XS Rating Curve= 0 ,0
Exp/Cntr(USF)=0,0
Exp/Cntr=0.3,0.1

Type RM Length L Ch R = 1 ,18106   ,2881.7,2881.7,2881.7
BEGIN DESCRIPTION:
HEC-2 RS: 180110
END DESCRIPTION:
XS GIS Cut Line= 6
2133198.10085543343084.9290509452136662.38825996337701.036504507
2136152.49314414334776.638046135  2134562.820136333831.832390353
2133308.94410524333570.6051741552132610.09220737333597.310031031
#Sta/Elev= 30
       0    8.43   205.4   10.95  1589.2    4.32  3365.2    5.78  3653.6    2.53
  3729.1    5.56  3789.7    1.75  4555.1    4.71  4632.8    1.95  5518.2    4.65
 10666.9    3.31 10849.1   -.75910977.39  -14.5411072.04  -14.54   11091   -.859
 11092.4    5.46   11121    1.56 11471.5    1.59 11491.6    5.25 11511.8    2.84
 12024.7    5.41 12051.6    2.65 12235.8    2.61 12286.1    8.74 12302.9    8.25
 12326.4   -1.25 12346.5   -1.72 12403.5    7.46 12523.7   11.5913200.33   11.28
#Mann= 3 ,-1,0
       0     .12       0 10849.1    .041       0   11091     .12       0
#XS Ineff= 1 ,-1
11097.4612249.01    5.48
Permanent Ineff=
       T
Bank Sta=10849.1,11091
XS Rating Curve= 0 ,0
Exp/Cntr(USF)=0,0
Exp/Cntr=0.3,0.1

Type RM Length L Ch R = 1 ,15225   ,,,
BEGIN DESCRIPTION:
HEC-2 RS: 177364 (LTR D)
END DESCRIPTION:
Node Name=D
XS GIS Cut Line= 6
2138686.88981973334170.621266617 2138072.9406002333078.175126334
 2135965.3590348332114.7867726172135877.29752476332038.207900614
2135718.47229846331890.3658788332134495.04402882331143.070104544
#Sta/Elev= 30
       0   12.11   447.2   10.41   624.7    7.63   846.8   11.68  1110.3     6.1
  1121.6     7.8  1308.9   13.22  1713.4    7.67  1784.6     2.3  1843.3     1.5
  2676.8    1.42  2763.4    3.01  2781.5    1.59  2907.8    2.73 3343.51     .96
 3458.03  -16.36 3572.96  -16.36  3617.8   1.161  3800.2    1.29  3873.3    8.34
  3938.2   10.46  3962.3    9.07  4043.1   10.81  4554.5    9.91  4694.9      12
  4754.6   10.65  5035.2    11.8  5063.3   10.06  5075.9   11.46  5337.8   11.34
#Mann= 3 ,-1,0
       0     .12       0 3343.51    .041       0  3617.8     .12       0
Bank Sta=3343.51,3617.8
XS Rating Curve= 0 ,0
Exp/Cntr(USF)=0,0
Exp/Cntr=0.3,0.1
LCMann Table=0

Chan Stop Cuts=-1
Use User Specified Reach Order=0
Composite Channel Slope=5

--- AshepooRiver.g04 (geometry) ---

Geom Title=Proposed Conditions
Program Version=6.60

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
River Reach=River 1         ,Reach 1

Type RM Length L Ch R = 1 ,61266   ,612.6,612.6,612.6
XS GIS Cut Line= 6
2109643.36416889348136.061039782 2109419.2208664346405.377529302
2108901.83713806345764.4344459052108097.35273658345035.840382716
2107248.48796725344541.4190195852105134.72207127343946.508637072
#Sta/Elev= 30
       0   24.82    27.9   26.11    54.4    24.4   223.1   23.32   319.1   20.59
   332.4   18.91   352.2   19.91   517.7   16.22   848.6   16.44    1110   13.88
  1148.9   11.68  1491.6      10  1655.7    5.29    19055.002243 1931.73   -1.28
 2027.04   -1.29    20555.025343  3262.9    5.26  3493.7    8.91  4618.7    10.3
  4885.3   13.88  4996.1   11.01  5013.1   13.05  5459.7   12.41  5568.8   14.07
  5752.9   13.87  5766.6    12.3  6090.5   15.56  6237.1   18.74  6837.5   21.14
#Mann= 3 ,0,0
       0     .12       0    1905    .041       0    2055     .12       0
#XS Ineff= 2 , 0
                            4079           10.03
Permanent Ineff=
       F       F
Bank Sta=1905,2055
XS Rating Curve= 0 ,0
Exp/Cntr(USF)=0,0
Exp/Cntr=0.5,0.3

Type RM Length L Ch R = 1 ,60653   ,910.6,910.6,910.6
XS GIS Cut Line= 5
2110712.77288746347311.8579898082109773.11276474345805.532602232
2108460.91386474344677.8068074582107503.50920049344364.812564901
2105104.22212249343861.947563075
#Sta/Elev= 30
       0   20.62    80.6   16.54   148.1   15.38   523.3   14.83   900.1   10.83
  1254.4      11  1393.6    8.63  1455.5    5.46 1543.58    4.65 1561.55   -1.27
 1668.17   -1.27    17004.898249  2040.4    6.18  2134.4     5.1  2965.2    5.12
  3130.8    7.38  3368.8    7.52  3734.8   10.32  4339.1    9.91  4840.4    14.4
  5031.2   12.07  5155.6   12.91  5172.3   11.43  5269.6   12.91  5564.6   13.05
  5742.4   15.36  6123.4   14.87  6315.7   18.45  6684.6   19.79  6964.3   23.76
#Mann= 3 ,0,0
       0     .12       0 1543.58    .041       0    1700     .12       0
#XS Ineff= 2 , 0
                            3179           10.03
Permanent Ineff=
       F       F
Bank Sta=1543.58,1700
XS Rating Curve= 0 ,0
Exp/Cntr(USF)=0,0
Exp/Cntr=0.5,0.3

Type RM Length L Ch R = 1 ,59743   ,692.5,692.5,692.5
XS GIS Cut Line= 6
 2111543.9979528346799.4654006252110720.29886494345621.270508605
2110432.87640412345334.4647799842109800.23240003344896.283538183
2108623.27742312  344521.24242642105070.32233361343764.748045568
#Sta/Elev= 30
       0   22.49   277.2   14.81   309.7   16.06   418.2   13.54   651.1   13.34
   849.8   10.38  1287.4   10.03  1423.1    6.79 1432.21    5.13  1474.9   -1.16
 1566.09   -1.16  1586.85.015964  2289.7    4.84  2396.2    6.32  2530.4    4.97
  3231.5    5.06  3703.4     7.6  3808.9    6.83  4147.1    9.62  4840.5   10.31
  5217.1   13.31  5673.7   12.59  5690.5   11.49  5700.5   12.56  5841.1   12.11
  6175.8   15.75  6456.9   14.12  6697.9   15.68  6888.7   19.12  7483.6   22.38
#Mann= 3 ,0,0
       0     .12       0 1432.21    .041       0  1586.8     .12       0
#XS Ineff= 2 , 0
             811   11.95    2429           10.03
Permanent Ineff=
       F       F
Bank Sta=1432.21,1586.8
XS Rating Curve= 0 ,0
Exp/Cntr(USF)=0,0
Exp/Cntr=0.5,0.3

Type RM Length L Ch R = 1 ,59050   ,254.1,254.1,254.1
BEGIN DESCRIPTION:
HEC-2 RS: 218448
END DESCRIPTION:
XS GIS Cut Line= 6
2112282.70593525346571.0636307492111510.76004851345480.860592143
2111131.56207502345054.5707431452110853.32104535344810.025185703
2110729.34134793344740.5849727232105051.66105604343662.589639585
#Sta/Elev= 30
       0   26.96   135.3   25.89     147   23.26   211.4   23.49   490.8   14.14
   685.9   14.54     806    11.2   891.1   12.22  1078.6    9.91  1434.1   10.93
  1763.5    4.68 1772.133.742357  1800.8   -1.35 1878.42   -1.35 1897.79    3.75
    1942    4.56  3846.3    5.41  3859.6    7.26  3882.9    5.81  4166.1    6.22
  5602.5   12.33    5753   10.69  6023.8   12.56  6388.3   12.31  6595.6    13.7
    6639   15.93  6679.2   14.03  6872.8   16.56  7156.3   14.34  8198.7   22.62
#Mann= 3 ,-1,0
       0     .12       0  1763.5    .041       0    1942     .12       0
#XS Ineff= 2 , 0
            1648   11.95    2062           10.03
Permanent Ineff=
       F       F
Bank Sta=1772.13,1897.79
XS Rating Curve= 0 ,0
Exp/Cntr(USF)=0,0
Exp/Cntr=0.5,0.3

Type RM Length L Ch R = 3 ,58980   ,,,
BEGIN DESCRIPTION:
S-15-41 over Ashepoo River
END DESCRIPTION:
Bridge Culvert--1,0,-1,-1, 0
Deck Dist Width WeirC Skew NumUp NumDn MinLoCord MaxHiCord MaxSubmerge Is_Ogee
53.74202,30,2.6,0, 73, 73, , , 0.98, 0, 2,2,,
       0     100     200     300     400     500     600     700     800     900
    1000    1100    1200    1300    1400    1500    1600    1700 1704.99    1705
 1774.99    1775    1935 1935.01    2005 2005.01    2100    2200    2300    2400
    2500    2600    2700    2800    2900    3000    3100    3200    3300    3400
    3500    3600    3700    3800    3900    4000    4100    4200    4300    4400
    4500    4600    4700    4800    4900    5000    5100    5200    5300    5400
    5500    5600    5700    5800    5900    6000    6100    6200    6300    6400
    6500    6600    6700
   25.38   24.71   23.63   22.11   19.99   18.13   16.17   14.93   13.88   13.31
   12.82   12.47   12.18   11.94   12.33   12.86   14.05   15.04   15.08   15.08
   15.59   15.59   15.55   15.55   15.01   15.01   14.44   13.06   12.03   11.54
   10.92   11.08   11.01   10.41   10.09   10.07   10.11   10.19   10.22   10.19
   10.12   10.28   10.02   10.18   10.16   10.05   10.21   10.23   10.26   10.58
   10.61   10.82   10.93   11.18   11.45   11.75   12.01   12.24   12.43    12.6
   12.98   13.29   13.36    13.6   13.77    13.9   14.01   14.19   14.29   14.42
    14.5   14.58   14.76
                                                                                
                                                                           11.78
   12.28   11.53   11.49   12.24    11.7
                                                                                
                                                                                
                                                                                
                                                                                
                        
      41     141     241     341     441     541     641     741     841     941
    1041    1141    1241    1341    1441    1541    1641    1741 1745.99    1746
 1815.99    1816    1976 1976.01    2046 2046.01    2141    2241    2341    2441
    2541    2641    2741    2841    2941    3041    3141    3241    3341    3441
    3541    3641    3741    3800    3900    4041    4141    4241    4341    4441
    4541    4641    4741    4841    4941    5041    5141    5241    5341    5441
    5541    5641    5741    5841    5941    6041    6141    6241    6341    6441
    6541    6641    6741
   25.38   24.71   23.63   22.11   19.99   18.13   16.17   14.93   13.88   13.31
   12.82   12.47   12.18   11.94   12.33   12.86   14.05   15.04   15.08   15.08
   15.59   15.59   15.55   15.55   15.01   15.01   14.44   13.06   12.03   11.54
   10.92   11.08   11.01   10.41   10.09   10.07   10.11   10.19   10.22   10.19
   10.12   10.28   10.02   10.18   10.16   10.05   10.21   10.23   10.26   10.58
   10.61   10.82   10.93   11.18   11.45   11.75   12.01   12.24   12.43    12.6
   12.98   13.29   13.36    13.6   13.77    13.9   14.01   14.19   14.29   14.42
    14.5   14.58   14.76
                                                                                
                                                                           11.78
   12.28   11.53   11.49   12.24    11.7
                                                                                
                                                                                
                                                                                
                                                                                
                        
Pier Skew, UpSta & Num, DnSta & Num=  ,1775, 2 ,1816, 2 , 0 , 0 , 0 ,,
       4       4
       3   12.28
       4       4
       2   12.28
Pier Skew, UpSta & Num, DnSta & Num=  ,1855, 2 ,1896, 2 , 0 , 0 , 0 ,,
       4       4
    -1.5   11.53
       4       4
    -1.7   11.53
Pier Skew, UpSta & Num, DnSta & Num=  ,1935, 2 ,1976, 2 , 0 , 0 , 0 ,,
       4       4
     4.5   12.24
       4       4
     4.5   12.24
Abutment Skew #Up #Dn= , 3 , 3
 1704.99    1707 1716.56
    9.78    9.78       5
 1745.99    1748 1757.56
    9.78    9.78       5
Abutment Skew #Up #Dn= , 3 , 3
 1993.59    2003 2005.01
       5     9.7     9.7
 2034.59    2044 2046.01
       5     9.7     9.7
BR Coef=-1 ,-1 ,-1 ,0.9, 0 ,,,0.8,0,1.2,0,
WSPro=,,,, 1 ,,,, 0 ,,,, 0 ,,,,-1 ,-1 ,-1 , 0 , 0 , 0 , 0 , 0
BC Design=,, 0 ,, 0 ,,,,,,
BC Use User HTab Curves=0
BC User HTab FreeFlow(D)= 0

Type RM Length L Ch R = 1 ,58796   ,616.6,616.6,616.6
BEGIN DESCRIPTION:
HEC-2 RS: 218419
END DESCRIPTION:
XS GIS Cut Line= 6
2112465.11983619 346422.549297062111363.13655015344933.468875854
2111165.40341921344740.6376676242110893.85305968344560.725925455
2110725.69108737 344502.288003772105210.34691174343461.561526106
#Sta/Elev= 30
       0   26.81    98.7   25.28   338.2   17.59     488    14.5   825.3   13.12
  1019.1    9.29  1282.2    9.85  1326.9   11.33  1352.7    9.53  1362.2   10.76
  1543.5    9.93 1812.413.262738 1833.62   -1.63 1922.08   -1.65  1943.2    3.23
  1980.2    4.55  2808.6    6.25  3565.2    5.26  4106.1    7.84  4356.5    6.81
  5294.1   10.04    5515   12.27  6482.5   12.12  6655.3    14.5  6902.9   13.88
  7204.5   15.59  7294.5   13.72  7978.7    19.6  8062.5   19.11    8247   22.13
#Mann= 3 ,-1,0
       0     .12       0 1812.41    .041       0  1980.2     .12       0
#XS Ineff= 2 , 0
            1661   11.95    2131           10.03
Permanent Ineff=
       F       F
Bank Sta=1812.41,1943.2
XS Rating Curve= 0 ,0
Exp/Cntr(USF)=0,0
Exp/Cntr=0.5,0.3

--- AshepooRiver.g05 (geometry) ---

Geom Title=Post Project
Program Version=6.60

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
River Reach=River 1         ,Reach 1
Reach XY= 30
2098396.23576606380646.8009591682097747.70079908376704.682944754
2098349.83399384 375176.529045482097726.69704407373600.953953826
2098114.75192337367841.6387006832099554.59564156365212.903242423
2099428.81121289363681.5771457152100708.15579364362482.324665464
2101289.63273322358523.8663055422100333.06655326351923.692230741
2105558.65619563 346752.098334352109100.83653268346361.782563958
 2111805.7756717  344595.11980812111881.37719572 342976.52674064
2110389.42873442341236.9377136342112009.03935508339315.330548813
2116615.76753564    339445.902442118850.12631383 341189.46406122
2121488.85557328  342010.05266182124117.63341542 340190.58593847
 2128091.1898635 340778.699006762130034.79235487  338498.5211566
2133356.08251692 338118.686337012134731.17271658 332679.67329194
2137633.21854056 330935.617395952135404.68988351 328442.04194944
 2135479.5315566 327368.052712862137781.44848433  324683.1006559
2139929.12472133 324531.725201252141596.00533789 322979.69654025

Type RM Length L Ch R = 1 ,88407   ,2944.8,2944.8,2944.8
XS GIS Cut Line= 4
2106397.55682745366319.4387589582101182.35958186366273.012670718
2095719.55653232366350.3894844512095038.64057147366396.815572691
#Sta/Elev= 30
       0   22.58    1045   22.71  1399.4   19.85  1422.4    17.1  1852.3   18.21
  2219.9   15.04    775015.87843 7766.29    6.58  7813.8    6.58    785015.78977
  7956.4   16.54  8031.9   24.97  8176.3   28.36  8572.5   30.41  8878.7   28.74
  9059.2   30.95    9289   26.94  9564.6   28.12  9725.5   29.23    9778   31.53
  9799.6   30.01  9886.4   30.88 10070.1   36.44 10339.2   39.94 10766.1   41.75
 11098.3   45.79 11259.5   43.14 11282.5   45.05 11305.6   41.84 11361.3   43.19
#Mann= 3 ,0,0
       0     .12       0    7750    .041       0    7850     .12       0
Bank Sta=7750,7850
XS Rating Curve= 0 ,0
Exp/Cntr(USF)=0,0
Exp/Cntr=0.3,0.1

Type RM Length L Ch R = 1 ,85462   ,2617.4,2617.4,2617.4
XS GIS Cut Line= 3
2106396.93542404363503.8041623472099505.29078866364086.196666745
  2095946.225484364798.009727677
#Sta/Elev= 30
       0   36.18   218.1   36.52   540.8   31.38     659   27.33  1169.9   24.49
  1713.3   18.15  1861.5    18.5  2154.6    13.7  2991.1   12.43  3350.1   13.96
  5408.5   12.88    687014.48625 6897.76    6.02 6956.29    6.02    697014.50333
  7867.4   15.06  8024.4      20  8456.1   20.75  8760.7   25.58  9554.2   32.22
    9801   31.71  9824.9   33.12  9881.8   28.22   10163      36 10236.6   36.79
 10253.3   33.72 10281.5   35.72 10310.2   33.46 10326.9   36.0510545.76   38.63
#Mann= 3 ,0,0
       0     .12       0    6870    .041       0    6970     .12       0
Bank Sta=6870,6970
XS Rating Curve= 0 ,0
Exp/Cntr(USF)=0,0
Exp/Cntr=0.3,0.1

Type RM Length L Ch R = 1 ,82845   ,2203.7,2203.7,2203.7
XS GIS Cut Line= 4
2106299.87000664362403.7294318162104876.24388478 362339.01915355
2100540.65524092362177.2434578832095687.38437094 363439.09388408
#Sta/Elev= 30
       0   35.25   728.1   21.25  2061.7    13.6  4636.3   12.21  5027.1    14.8
  5139.1   12.735586.82113.15396 5625.24    5.37 5672.39    5.375686.82113.30377
  7498.9   12.78  7631.1   17.12  7651.4   14.98  7787.1   15.77  7834.6   18.72
    7963   17.76  8268.2   23.02  8458.1   21.98  8654.8   24.44    8787   22.93
  8833.9    25.5  8915.9   24.42  9092.2   27.09 10041.7   27.26 10055.2   23.98
 10065.4   25.71 10129.8   26.32 10431.6    27.2 10638.5   26.5810778.33   23.46
#Mann= 3 ,0,0
       0     .12       05586.821    .041       05686.821     .12       0
Bank Sta=5586.821,5686.821
XS Rating Curve= 0 ,0
Exp/Cntr(USF)=0,0
Exp/Cntr=0.3,0.1

Type RM Length L Ch R = 1 ,80641   ,1673.9,1673.9,1673.9
XS GIS Cut Line= 4
2106043.70142807 360642.752451782101182.44207423 360642.75245178
 2100503.1394571360557.8396246392095535.73906933362065.042306397
#Sta/Elev= 30
       0   44.15   441.6   32.28   500.7   27.65     819   21.02  1787.2   13.09
  2151.4   15.38  2328.7   13.34  2548.5    14.1    2834   16.94  3145.8   24.44
  3342.7   22.02  3519.9   17.17  3585.6   12.88  3726.7   11.355170.20611.55534
 5193.38    4.86 5241.73    4.865270.20611.58589  6414.5   13.53  7511.9   11.97
  8427.2   13.66  8471.8   15.87  8492.4   13.91  8533.5    16.6  8554.1   14.14
  9034.8   14.75  9397.8   19.33 10035.7   21.45 10207.1   24.76 10736.9   28.99
#Mann= 3 ,0,0
       0     .12       05170.206    .041       05270.206     .12       0
Bank Sta=5170.206,5270.206
XS Rating Curve= 0 ,0
Exp/Cntr(USF)=0,0
Exp/Cntr=0.3,0.1

Type RM Length L Ch R = 1 ,78967   ,1132.2,1132.2,1132.2
XS GIS Cut Line= 4
2105258.25777701358201.5086714672101882.97289815358902.039495383
 2100205.9445621359411.5164582312095302.22879469360748.893485707
#Sta/Elev= 30
       0   24.01   838.7   14.36  1247.6   16.93  2028.6   11.69  2219.6   15.75
  2923.5   16.96  3208.4   15.74  3335.7   11.534141.57110.59565 4173.95     4.4
 4220.34     4.44241.57110.63325  5790.9   11.51  5974.6    14.6    6012   11.81
  6175.2   11.34  6318.1   13.82  6362.3   10.73  6406.4   13.81  6556.2   10.78
    6580   13.35    6995   11.38  7013.6   14.33  7062.7   11.57  7460.7    11.5
  9372.4   16.62    9784   23.85  9855.4   22.74 10151.4   34.7210282.74   36.63
#Mann= 3 ,0,0
       0     .12       04141.571    .041       04241.571     .12       0
Bank Sta=4141.571,4241.571
XS Rating Curve= 0 ,0
Exp/Cntr(USF)=0,0
Exp/Cntr=0.3,0.1

Type RM Length L Ch R = 1 ,77835   ,817.9,817.9,817.9
XS GIS Cut Line= 4
 2104111.9346106357522.2060543372099845.06504675358350.106118965
2096108.90065254358923.2677021682094813.98003863359284.147217519
#Sta/Elev= 30
       0   22.58   417.7   21.22   835.5   14.74   978.3   14.84  1109.7   10.85
    1474   14.72  2473.6   19.15  2577.2   17.97  2654.1   11.31    303511.03299
  3071.3       4 3119.82    3.99    313510.11057    4242    9.92  4448.6   11.92
  4823.7    10.4  4976.5   12.92    5252   10.28  5414.3   11.96    6222   10.22
  7748.4   13.19  7897.9   15.31  7984.2   15.19  8004.1   13.07  8077.2   16.18
    8161   14.55  8668.7   17.76  9125.3   17.44  9407.9   24.949470.586   24.36
#Mann= 3 ,0,0
       0     .12       0    3035    .041       0    3135     .12       0
Bank Sta=3035,3135
XS Rating Curve= 0 ,0
Exp/Cntr(USF)=0,0
Exp/Cntr=0.3,0.1

Type RM Length L Ch R = 1 ,77017   ,1190.2,1190.2,1190.2
XS GIS Cut Line= 4
2103719.85250626357044.0968831052100627.32658961357379.108622936
2095876.54498006358231.4916030132095024.16199999358432.052304208
#Sta/Elev= 30
       0   19.67   480.2   18.26   734.3   10.75  1477.1   12.01  1701.5   16.53
  2015.1   17.68  2236.3   15.38  2348.5   12.25  2546.6   12.99  2681.9     9.4
    273510.22525  2751.7    3.58 2810.91    3.59    283510.08146  3457.8    9.25
  4638.1   11.42  5724.7   10.07  5805.5    11.4  5911.4    9.63  5932.7   11.33
  6948.3   11.55  7258.4   17.95  7538.5    15.5  7708.5   16.07  7738.5   17.78
  7866.4   15.39  8235.3   14.52  8252.1   15.96  8636.5   16.338812.922   18.76
#Mann= 3 ,0,0
       0     .12       0    2735    .041       0    2835     .12       0
Bank Sta=2735,2835
XS Rating Curve= 0 ,0
Exp/Cntr(USF)=0,0
Exp/Cntr=0.3,0.1

Type RM Length L Ch R = 1 ,75827   ,952.8,952.8,952.8
XS GIS Cut Line= 6
2103484.77253227356585.643760793 2102409.3881305356342.559731688
2101850.75576887356271.4910918842101200.12087369356311.763392387
2097028.31291086356773.2007179292096279.54032397356915.172039683
#Sta/Elev= 30
       0   19.62    31.9   18.77      60   22.22    73.5   19.87   110.5   18.75
   466.4   17.22   655.5   18.92   800.2   15.89  1092.9   15.52  1271.7   12.33
  1301.5   13.68    1318   10.01  1347.8    9.25  1552.9    9.22  1589.3   10.83
  1665.4     9.1  2050.1   10.56    2277    9.21  2372.6   10.87    26759.566566
 2706.35    3.13 2784.84    3.13    28059.734908  6506.2   10.83  6786.7   15.92
  7177.5   16.54  7187.5   17.61  7204.2   24.26  7220.9   17.18  7277.1   16.59
#Mann= 3 ,0,0
       0     .12       0    2675    .041       0    2805     .12       0
Bank Sta=2675,2805
XS Rating Curve= 0 ,0
Exp/Cntr(USF)=0,0
Exp/Cntr=0.3,0.1

Type RM Length L Ch R = 1 ,74874   ,811.4,811.4,811.4
XS GIS Cut Line= 6
2103563.33853893356122.9023916632102439.46191877355741.479447767
2100828.15808317355532.0491173452099585.11723442355535.141277814
2097678.49577922355601.6040459542096639.78637301355746.062602483
#Sta/Elev= 30
       0   22.29   325.8   20.18   643.8   21.37  1122.1    17.8  1402.5   11.09
  1597.9   10.61  1657.9   12.43  1991.3    8.67  2417.9   10.17 2852.64    8.56
 2870.41    2.71 2994.83    2.71    30158.550438  3407.7    8.66  3529.1   11.41
  3617.7    9.44  3962.3   12.21  4159.2    8.89  4658.4    9.84  4674.8   11.53
  4904.7    8.88  5416.6   11.17  5600.5     9.8  5774.5   11.88  5830.3   10.05
  6067.7   20.02  6325.2   18.09  6432.2   19.89  6458.7   18.05  7012.1   18.06
#Mann= 3 ,0,0
       0     .12       0 2852.64    .041       0    3015     .12       0
Bank Sta=2852.64,3015
XS Rating Curve= 0 ,0
Exp/Cntr(USF)=0,0
Exp/Cntr=0.3,0.1

Type RM Length L Ch R = 1 ,74063   ,1021,1021,1021
XS GIS Cut Line= 6
2103682.61513281355697.0549044052102284.70829131355122.464937907
2100677.49266574354792.8194410942099999.66209378354803.752192255
2097708.15364479354935.6286455442096807.74356719 355079.52451163
#Sta/Elev= 30
       0   24.47   343.8   24.75   747.2   22.27  1305.9   10.01  1703.3   11.07
  2210.3    8.92  2468.9    9.23  2482.3   10.92  2499.1    8.64    29558.099456
 2985.25    2.41 3071.13     2.4 3098.528.422089  3330.9    8.16  3396.7   10.41
  3672.3    8.82  4438.2    10.1  4655.3    8.51  4928.1   10.62  5552.2    9.34
  5604.7   11.17  5956.4    9.55  6114.1   11.19  6210.4   15.81  6233.6   13.26
  6366.6   17.02  6413.3   16.31    6443   18.29  6672.3    17.4  7037.4   19.26
#Mann= 3 ,0,0
       0     .12       0    2955    .041       0 3098.52     .12       0
Bank Sta=2955,3098.52
XS Rating Curve= 0 ,0
Exp/Cntr(USF)=0,0
Exp/Cntr=0.3,0.1

Type RM Length L Ch R = 1 ,73042   ,702.4,702.4,702.4
XS GIS Cut Line= 6
2104580.48483008 355241.062238682101661.80877761353965.224877458
2101171.16157919353868.206247267 2100082.3226075354092.234792296
2097823.82905937354594.7347783322096794.35129549 354866.19170869
#Sta/Elev= 30
       0   18.77  1135.9   10.47  1383.4   10.12    1492   12.69  1626.4      13
  1796.9   11.55  1882.8    9.16  2022.9   11.57    2195    9.14  2619.6    11.4
  3045.7    8.72    3418    8.82  3428.5   10.08  3582.4    7.91    3870 8.34008
 3920.28    1.88 4015.14    1.88 4039.05    8.19  5507.9    9.62    6029    8.24
  6150.1    10.3  6694.3    9.44  6912.9   10.92  7000.3    9.24  7162.1   12.13
  7179.1   10.33  7219.8   13.17    7626   18.08  7815.1   17.03  8175.6   18.93
#Mann= 3 ,0,0
       0     .12       0    3870    .041       0 4039.05     .12       0
Bank Sta=3870,4039.05
XS Rating Curve= 0 ,0
Exp/Cntr(USF)=0,0
Exp/Cntr=0.3,0.1

Type RM Length L Ch R = 1 ,72340   ,1313.4,1313.4,1313.4
XS GIS Cut Line= 6
2104641.45660154354877.0331971342101692.11568816353517.983834757
2100893.78222901353339.0597686792099760.68197156  353489.0289204
2098619.17759005 353758.006675212096722.45335365354443.507094647
#Sta/Elev= 30
       0   20.23     398   18.24   566.7   15.36   846.7   14.94  1161.5   10.63
    1449   12.43  1764.3    9.81  2491.9    9.13  2717.6   11.65  3068.8   12.11
  3240.8   11.33  3352.3    8.63  3883.7    7.62  4101.7   10.79  4171.3    8.19
    43307.960487 4368.31    1.61 4458.54    1.63 4485.35    7.91    5784     7.5
  5922.2    9.02  5972.8    7.53  6435.8   10.12  7063.4    9.32  7084.3   12.07
  7137.8    9.71  7540.5    8.97  7726.5    9.66  7985.9   15.38  8399.6      15
#Mann= 3 ,0,0
       0     .12       0    4330    .041       0 4485.35     .12       0
Bank Sta=4330,4485.35
XS Rating Curve= 0 ,0
Exp/Cntr(USF)=0,0
Exp/Cntr=0.3,0.1

Type RM Length L Ch R = 1 ,71026   ,932,932,932
XS GIS Cut Line= 6
2104500.83237574354502.2540987692102059.37782849353224.823799985
2100860.60817398352609.7235453542100308.18738998352348.740765757
2099630.38953622351822.9891955322098164.55244227350216.185473509
#Sta/Elev= 30
       0   19.48   632.4   18.27   947.2    13.9  1006.5   10.88  1258.3    9.94
  2033.5    9.06  2502.8   14.52  2699.1   11.66  3237.4    15.8  3399.9   10.39
  3650.8     8.4  4794.8     7.4 4813.52    1.17  4926.2    1.17  4958.17.728683
  6900.1    7.63  6925.6   10.19  6971.1     8.1  7085.2   10.27  7153.2   15.68
  7231.3   16.27  7259.9   18.94  7294.6   14.71  7374.6   13.88  7387.9   14.32
  7405.7   18.69  7423.5   16.76  7481.2   20.38  7639.7   22.06  7747.3   19.81
#Mann= 3 ,0,0
       0     .12       0  4794.8    .041       0  4958.1     .12       0
Bank Sta=4794.8,4958.1
XS Rating Curve= 0 ,0
Exp/Cntr(USF)=0,0
Exp/Cntr=0.3,0.1

Type RM Length L Ch R = 1 ,70094   ,659,659,659
XS GIS Cut Line= 4
2104436.01786635354160.1425241452102459.03756485352876.263836931
2100652.50396726351583.2095389232098728.33976301 349899.56586021
#Sta/Elev= 30
       0   21.16   602.7   19.06   879.8   14.49  1111.3   13.75  1440.2    9.69
  2351.7   11.27  2476.7   15.47  2908.5   18.53  3005.4   17.15  3099.1   10.94
  3203.1     9.6  3269.6    6.42  4333.2    7.16 4375.27     .87 4473.31     .88
    44957.172149  4718.3    7.01  4897.7    11.1  5011.1   17.19  5220.8   18.94
  5364.8   17.27  5455.9   10.72  5547.5    8.43  6293.2    7.68  6476.3   11.71
    6690   25.91  6764.2   28.39  6913.8   39.29  7038.9   39.15  7135.7   36.27
#Mann= 3 ,0,0
       0     .12       0  4333.2    .041       0    4495     .12       0
Bank Sta=4333.2,4495
XS Rating Curve= 0 ,0
Exp/Cntr(USF)=0,0
Exp/Cntr=0.3,0.1

Type RM Length L Ch R = 1 ,69435   ,1039,1039,1039
XS GIS Cut Line= 5
 2104668.4043109353865.4570101392103846.66691624353225.991559639
2102131.87292103351894.7699054612101242.87252992351244.294252948
 2099285.9100722349593.448827716
#Sta/Elev= 30
       0   29.01   343.8   27.99   814.2   14.66   879.3   16.53   925.7   14.34
  1099.2    15.1  1267.3   10.01  2274.1      11  2488.7   16.42  2812.8   18.72
  3045.5   17.87  3178.6   10.47  3329.6   10.34  3455.6       7    42156.777931
 4241.53     .65 4337.39     .65    43656.781381  4840.6    8.41  4953.4   13.54
    5151   17.22  5276.8   16.32  5500.4    8.96  6072.3   10.55  6177.1   15.66
  6284.4   14.96  6490.5   21.72  6632.2   43.97  6754.4   46.95  6873.9   45.49
#Mann= 3 ,0,0
       0     .12       0    4215    .041       0    4365     .12       0
Bank Sta=4215,4365
XS Rating Curve= 0 ,0
Exp/Cntr(USF)=0,0
Exp/Cntr=0.3,0.1

Type RM Length L Ch R = 1 ,68396   ,842,842,842
XS GIS Cut Line= 3
2104785.08390592353190.3239595122101855.10659491350457.136169394
2099777.88387442348926.551006928
#Sta/Elev= 30
       0   40.19   183.1   37.64   336.3   27.32   652.1   12.66   772.2   10.92
  1742.9   10.27  1760.9   10.82  1778.3   16.86    1797   10.74  1832.7   10.38
  1855.1   16.38  1883.6   12.38  2402.9   17.78    2663   15.66  2761.7    8.77
    38756.639429 3890.62    .372 4012.31    .372    40256.689871  4636.9     7.9
  4665.5   10.67  4678.7    7.02  5166.9    6.91  5179.1   10.92  5272.9    9.32
    5546   15.01  5835.4   15.84  6122.2    31.1  6430.6   32.17  6587.1   37.07
#Mann= 3 ,0,0
       0     .12       0    3875    .041       0    4025     .12       0
Bank Sta=3875,4025
XS Rating Curve= 0 ,0
Exp/Cntr(USF)=0,0
Exp/Cntr=0.3,0.1

Type RM Length L Ch R = 1 ,67554   ,483.1,483.1,483.1
XS GIS Cut Line= 3
2105036.53718261352753.0139130932102423.60965525349877.700357889
2100444.78169521348368.980697743
#Sta/Elev= 30
       0   39.62     195   38.67   231.7   36.44   353.6   33.53   599.9   19.85
   751.3   14.96   814.7   10.86  1120.3    9.37    1537   10.56  1606.4    8.98
  1766.1   11.18  1917.6   11.35  2065.9    14.6    2103   13.59  2214.6   14.54
  2382.4   12.86  2458.5    9.56  2635.1   10.21    3118    6.25    37756.143803
 3789.86      .1 3912.11     .15    39256.251347  5428.5    8.56  5552.2   10.14
  5624.8   14.06  5657.6    17.5  5891.7   26.46  6072.6   30.37  6373.6   29.37
#Mann= 3 ,0,0
       0     .12       0    3775    .041       0    3925     .12       0
Bank Sta=3775,3925
XS Rating Curve= 0 ,0
Exp/Cntr(USF)=0,0
Exp/Cntr=0.3,0.1

Type RM Length L Ch R = 1 ,67071   ,535.9,535.9,535.9
XS GIS Cut Line= 3
2105016.33473616351978.5532578462102532.84558371349346.594645189
2100845.69262688347902.391714141
#Sta/Elev= 30
       0   25.76     133   21.84   152.1   19.44   232.3   13.53   324.3   13.51
   383.2   11.44   637.4   11.48   689.7    10.2     887     9.2   924.2   10.38
   942.7    9.07  1503.8    8.82  1922.4   12.05  1993.2   11.75  2067.8    9.97
  2480.9     8.4  2495.3    9.07  2558.6    6.87  2605.2    6.47    33006.612388
    3315    -.03    3435    -.03    34506.212595  3902.8    6.12  4573.7    8.72
  4962.6   14.72  5282.2   24.06  5429.1   24.57  5588.9   22.95  5839.5   25.53
#Mann= 3 ,0,0
       0     .12       0    3300    .041       0    3450     .12       0
Bank Sta=3300,3450
XS Rating Curve= 0 ,0
Exp/Cntr(USF)=0,0
Exp/Cntr=0.3,0.1
