HEC-RAS study WillowCreek.prj: S-21-57 over Willow Creek

--- WillowCreek.g02 (geometry) --- (continued)

Type RM Length L Ch R = 1 ,142882  ,600,600,600
BEGIN DESCRIPTION:
Willow Creek 35.0
END DESCRIPTION:
XS GIS Cut Line= 3
      2419676.32       827426.47      2420363.93       826543.79
      2421143.68        825207.1
#Sta/Elev= 30
  3881.1   79.17  4315.8   60.96  4754.7   59.19  4840.5   47.81  4853.6   43.03
  4939.4   47.75  4971.1      47  4972.7   46.64  4974.9    41.7  4975.4    40.7
  5025.1    41.7  5025.3   44.33    5026   42.06  5032.2   42.24    5046   46.48
    5060   47.01  5112.1   45.27  5139.7    41.7  5174.2    46.1  5266.9   42.25
  5290.8   47.43  5508.3   43.14  5577.6   44.46  5630.2   49.34  5905.2   48.26
  6091.4   55.18  6135.3   59.14  6209.8   71.19  6294.7   73.23  6547.5   72.54
#Mann= 3 ,0,0
  3881.1     .12       0  4974.9     .04       0  5025.1     .12       0
Bank Sta=4974.9,5025.1
XS Rating Curve= 0 ,0
Exp/Cntr=0.3,0.1

Type RM Length L Ch R = 1 ,142282  ,900,900,900
BEGIN DESCRIPTION:
Willow Creek 34.0
END DESCRIPTION:
XS GIS Cut Line= 4
      2420367.23       828141.77      2420781.44       826626.71
      2420789.18       826492.09      2421180.38       825341.58
#Sta/Elev= 30
  3294.5   70.67  3563.3   63.91    3606   65.08    3715   60.35  3785.7   60.76
  3836.5   57.15  3901.9   57.76  4012.9   48.77    4090   46.82    4570   48.07
  4669.6   47.17  4702.7    42.6    4768   41.12  4908.5   46.02  4937.2   42.09
  4948.7   44.51  4974.9   41.12  4975.4   40.12  5025.1   41.12  5027.2   46.47
  5173.9   42.08  5200.1   45.91  5296.1   47.07  5695.5   51.09  5704.3   47.87
  5716.1   51.14  5736.9   49.74  5913.3   56.92  5925.6   60.18  6215.2   70.62
#Mann= 3 ,0,0
  3294.5     .12       0  4974.9     .04       0  5025.1     .12       0
Bank Sta=4974.9,5025.1
XS Rating Curve= 0 ,0
Exp/Cntr=0.3,0.1

Type RM Length L Ch R = 1 ,141382  ,500,500,500
BEGIN DESCRIPTION:
Willow Creek 32.0
END DESCRIPTION:
XS GIS Cut Line= 3
      2420538.39        828166.3      2421415.78       826308.57
       2421834.6       825946.85
#Sta/Elev= 30
  2945.5   69.82  2986.6   65.61    3033   68.93  3356.5   58.27  3753.5   55.54
  4044.6   45.19  4473.5   46.65  4607.5   42.05  4652.1   45.06  4736.3   42.09
  4764.7   43.01  4769.1   45.66    4787   42.95  4863.5   42.16  4949.9   42.13
  4966.6   44.69    4972   44.09  4974.9      41  4975.4      40  5025.1      41
  5025.6   43.93  5034.7   46.36  5076.2   47.99  5227.3   46.25  5276.2   52.64
  5325.9    64.1  5366.6   76.49  5405.3   82.47  5462.9   85.78  5553.4   85.28
#Mann= 3 ,0,0
  2945.5     .12       0  4974.9     .04       0  5025.1     .12       0
Bank Sta=4974.9,5025.1
XS Rating Curve= 0 ,0
Exp/Cntr=0.3,0.1

Type RM Length L Ch R = 1 ,140882  ,500,500,500
BEGIN DESCRIPTION:
Willow Creek 31.0
END DESCRIPTION:
XS GIS Cut Line= 3
      2420672.91       828257.98      2421844.89       826441.31
      2422034.15       826250.01
#Sta/Elev= 30
  2838.1      76  2897.1   75.74  3028.7   68.07  3243.6   59.65  3350.2    58.6
    3373   56.49  3451.6    57.5  3765.2   52.97  3776.2   51.39  4018.2   51.87
  4096.1   46.13  4144.6   44.94  4345.8   45.25  4372.2   43.25  4403.6    45.8
  4549.4   46.16  4593.8   42.56  4744.3    41.8  4811.7   43.71  4871.1   41.57
  4957.2   42.22  4974.9   40.53  4975.4   39.53  5025.1   40.53  5025.7    46.9
  5030.9   49.98  5045.8   58.11  5082.2   72.37    5150   81.61  5269.1   83.04
#Mann= 3 ,0,0
  2838.1     .12       0  4974.9     .04       0  5025.1     .12       0
Bank Sta=4974.9,5025.1
XS Rating Curve= 0 ,0
Exp/Cntr=0.3,0.1

Type RM Length L Ch R = 1 ,140382  ,800,800,800
BEGIN DESCRIPTION:
Willow Creek 30.0
END DESCRIPTION:
XS GIS Cut Line= 3
      2420954.17       828388.81      2422130.99        826825.8
      2422213.82       826473.92
#Sta/Elev= 30
  3043.5   83.86  3137.6   80.28  3270.4   72.76  3277.7   70.98  3286.6   71.98
  3380.1   64.84  3692.1   54.92    3970   50.31  3987.4   51.69  4206.2   49.93
    4258   47.45  4372.1   48.36  4520.4   44.98  4534.5   43.07  4619.2   44.11
  4645.2   42.27  4688.5   44.97  4768.7   44.61  4974.9   40.03  4975.4   39.03
  5025.1   40.03  5150.8    42.4  5153.6    43.9  5179.3   44.52  5196.4   46.85
    5220   53.67  5263.7   71.13  5308.5   77.33  5333.5   78.23  5361.5   76.58
#Mann= 3 ,0,0
  3043.5     .12       0  4974.9     .04       0  5025.1     .12       0
Bank Sta=4974.9,5025.1
XS Rating Curve= 0 ,0
Exp/Cntr=0.3,0.1

Type RM Length L Ch R = 1 ,139582  ,500,500,500
BEGIN DESCRIPTION:
Willow Creek 29.0
END DESCRIPTION:
XS GIS Cut Line= 3
      2421129.85       828426.65      2422541.39         827337.
      2423797.17       826719.69
#Sta/Elev= 30
  3216.8   82.89  3360.7   74.31  3401.2   69.24  3571.6   63.08  3593.1   64.73
  3608.7   62.49  3747.8   57.15  3921.2   53.24  3972.4   47.65    4648   45.56
  4863.2   43.39  4972.5   39.03    4973   38.03  5027.5   39.03  5141.9   40.56
  5175.3   44.07  5452.4   45.52  5530.7    49.3  5609.5   48.25  6007.2   51.08
  6098.8   56.93  6179.4   68.66  6190.1    66.8  6198.8   68.92  6205.6   66.82
  6227.2   69.57  6250.3   75.93  6294.8    80.5  6326.6      87  6399.3   90.84
#Mann= 3 ,0,0
  3216.8     .12       0  4972.5     .04       0  5027.5     .12       0
Bank Sta=4972.5,5027.5
XS Rating Curve= 0 ,0
Exp/Cntr=0.3,0.1

Type RM Length L Ch R = 1 ,139082  ,600,600,600
BEGIN DESCRIPTION:
Willow Creek 28.0
END DESCRIPTION:
XS GIS Cut Line= 3
      2421210.98       828639.47      2422715.75       827709.41
      2424046.46       826868.39
#Sta/Elev= 30
    3231   85.68  3413.2   80.43  3538.4   71.51  3539.5   72.96  3647.1    69.8
  3913.4   54.68  3920.9   52.33  4044.5   49.06  4114.4   44.44  4133.7   45.62
  4164.7   43.39  4262.3      46  4313.4   43.19  4636.6   43.76  4697.9   42.44
  4724.8   39.08  4968.6   40.57  4972.5   38.86    4973   37.86  5027.5   38.86
  5028.5   45.96  5049.4   50.24  5617.3   50.16  5711.7   48.44  5869.6   50.09
  6079.7   59.17    6278   81.88    6309   80.13    6351   84.77  6574.2   90.72
#Mann= 3 ,0,0
    3231     .12       0  4972.5     .04       0  5027.5     .12       0
Bank Sta=4972.5,5027.5
XS Rating Curve= 0 ,0
Exp/Cntr=0.3,0.1

Type RM Length L Ch R = 1 ,138482  ,400,400,400
BEGIN DESCRIPTION:
Willow Creek 27.0
END DESCRIPTION:
XS GIS Cut Line= 3
      2421455.49       828755.67      2422535.62       828111.75
      2424280.21       827129.31
#Sta/Elev= 30
  3742.5   78.41  3868.8   70.06  3946.5   70.79  4107.7   65.77  4330.5   49.64
  4566.9   44.76    4710   47.66  4828.1    43.4  4867.1    39.9  4930.9   41.08
  4972.5   37.93    4973   36.93  5027.5   37.93    5036    39.8  5075.8   39.99
  5158.4   38.29  5204.6   42.88  5380.9   47.49  5432.9   45.45  5567.3   50.46
  5635.3   48.12  5671.8   43.16  5728.9   46.67  5960.7   44.09  6056.6   48.76
  6143.3   48.82  6433.6   60.88  6462.1    59.3  6679.9   66.57  7002.2   82.31
#Mann= 3 ,0,0
  3742.5     .12       0  4972.5     .04       0  5027.5     .12       0
Bank Sta=4972.5,5027.5
XS Rating Curve= 0 ,0
Exp/Cntr=0.3,0.1

Type RM Length L Ch R = 1 ,138082  ,600,600,600
BEGIN DESCRIPTION:
Willow Creek 26.0
END DESCRIPTION:
XS GIS Cut Line= 3
      2421810.12       829201.99      2422795.24       828304.43
      2424310.81       827257.69
#Sta/Elev= 30
  3667.3   83.09  3783.9   76.41    3920   64.89  4106.2   57.74  4278.3   45.99
    4474   45.79  4530.8   42.42  4555.3   44.52  4620.5    42.3  4678.5   44.98
    4858    39.1  4940.7   41.88  4948.2   38.64  4972.5   38.44    4973   35.19
    5027   35.19  5027.5   38.44  5057.3   42.28    5190   45.42  5479.2   47.22
  5797.7   43.06  6063.6   49.31  6159.6   56.29  6377.6   59.18  6480.1   63.66
  6605.1   72.53  6632.6   71.52  6657.9      75  6738.1   76.17  6841.9   83.88
#Mann= 3 ,0,0
  3667.3     .12       0  4972.5     .04       0  5027.5     .12       0
Bank Sta=4972.5,5027.5
XS Rating Curve= 0 ,0
Exp/Cntr=0.3,0.1

Type RM Length L Ch R = 1 ,137482  ,600,600,600
BEGIN DESCRIPTION:
Willow Creek 25.0
END DESCRIPTION:
XS GIS Cut Line= 3
      2421950.79       829116.37      2422985.01       828693.84
      2424390.29       827752.93
#Sta/Elev= 30
  3882.8   70.71  4042.7   60.13  4258.6   58.37  4346.9   46.46  4484.7   47.89
  4531.7   41.83  4644.6   44.94    4890      43  4916.8   39.27  4972.5   38.39
    4973   35.67    5027   35.67  5027.5   38.39  5040.2    41.7  5071.1   38.81
    5087   42.12  5160.8   39.48  5231.2   41.63  5325.4   39.43  5364.6   43.75
  5469.4   41.67  5537.5   43.48    5586   40.68  5702.8   46.84  6111.9   43.47
  6190.3   52.29  6236.3   65.92  6260.7   69.11  6558.9   69.03  6691.2    71.3
#Mann= 3 ,0,0
  3882.8     .12       0  4972.5     .04       0  5027.5     .12       0
Bank Sta=4972.5,5027.5
XS Rating Curve= 0 ,0
Exp/Cntr=0.3,0.1

Type RM Length L Ch R = 1 ,136882  ,500,500,500
BEGIN DESCRIPTION:
Willow Creek 24.0
END DESCRIPTION:
XS GIS Cut Line= 4
      2421944.66       829305.91      2423186.48       828927.49
      2423297.84       828913.94      2424640.92       828333.79
#Sta/Elev= 30
  3701.8   75.64  3958.3   52.48  4210.5   51.65  4504.9   45.53  4652.5    47.3
  4861.5   44.84  4883.7   43.76  4905.4    38.7  4972.5   37.75    4973   35.21
    5027   35.21  5027.5   37.75  5030.9   40.41    5083   38.89  5101.1   41.29
  5280.1   38.03  5306.6   43.48  5391.7   40.24  5434.8    43.7  5480.5   40.72
  5513.8   43.25  5602.7   41.27  5701.2   45.14  6022.3   42.92  6241.7   44.89
  6281.6   47.46  6386.7   45.48  6433.2   48.46  6532.8   65.96  6575.2   67.84
#Mann= 3 ,0,0
  3701.8     .12       0  4972.5     .04       0  5027.5     .12       0
Bank Sta=4972.5,5027.5
XS Rating Curve= 0 ,0
Exp/Cntr=0.3,0.1

Type RM Length L Ch R = 1 ,136382  ,500,500,500
BEGIN DESCRIPTION:
Willow Creek 23.0
END DESCRIPTION:
XS GIS Cut Line= 3
      2421926.31       829354.83      2423480.83       829120.35
      2424879.34       829104.15
#Sta/Elev= 30
  3427.9   78.73  3655.8   56.43  3766.7   51.64  4069.1   50.47  4188.5   47.55
  4383.5   48.85  4472.7   46.23  4580.1   47.96  4677.7   44.45  4851.4   44.08
  4884.6   38.52  4972.5   37.58    4973   34.73    5027   34.73  5027.5   37.58
  5042.9   41.66  5101.3    37.7  5207.7   40.38  5242.4   39.14  5267.8   42.24
  5365.3   43.72  5496.3   41.88  5661.3   42.58  5766.3   46.21  5861.1   44.62
  6135.5   46.46  6149.7   50.11  6193.8   54.06  6279.3    71.7  6398.6    75.6
#Mann= 3 ,0,0
  3427.9     .12       0  4972.5     .04       0  5027.5     .12       0
Bank Sta=4972.5,5027.5
XS Rating Curve= 0 ,0
Exp/Cntr=0.3,0.1

Type RM Length L Ch R = 1 ,135882  ,600,600,600
BEGIN DESCRIPTION:
Willow Creek 22.0
END DESCRIPTION:
XS GIS Cut Line= 3
      2421865.19       829415.97      2423613.29       829486.06
      2424995.52       829660.53
#Sta/Elev= 30
  3250.5   81.97  3359.9   71.24  3704.2   53.04  3891.6   54.31  4026.9   46.14
  4262.7   48.89  4479.6   44.17  4659.8   45.68  4740.4   40.62  4790.9   43.47
  4913.8   42.12  4933.1   38.08  4962.4   39.88  4972.5    37.5    4973   34.85
    5027   34.85  5027.5    37.5    5034    40.8  5062.5   38.89  5098.3   43.19
    5230   40.75  5600.6   45.89  5724.5   43.53  5788.2   49.01  5916.3    74.3
  5982.4   79.75  6048.9   80.98    6182   75.47  6277.5   84.49  6393.2   89.69
#Mann= 3 ,0,0
  3250.5     .12       0  4972.5     .04       0  5027.5     .12       0
Bank Sta=4972.5,5027.5
XS Rating Curve= 0 ,0
Exp/Cntr=0.3,0.1

Type RM Length L Ch R = 1 ,135282  ,400,400,400
BEGIN DESCRIPTION:
Willow Creek 21.0
END DESCRIPTION:
XS GIS Cut Line= 4
      2421718.46       829703.33      2423454.75       829803.89
      2423610.47       829841.47      2424781.55       829850.06
#Sta/Elev= 30
  3260.8   84.23  3397.9   79.29  3570.2   64.58  3724.1   59.38  4055.7   56.92
  4286.8    49.1  4386.8   51.29  4780.5   50.06  4972.5   37.26    4973   34.08
    5027   34.08  5027.5   37.26  5057.3   40.08  5106.8   37.86  5130.9   41.41
    5167   42.09  5244.7   41.02  5257.2    38.1  5410.7   38.01  5469.2   38.42
  5527.5   42.29    5609   38.69  5649.7   42.19  5725.1   39.97  5881.1    42.9
  5971.1   47.49  6026.1   54.07  6110.2   73.58  6183.8   82.69  6331.3   89.24
#Mann= 3 ,0,0
  3260.8     .12       0  4972.5     .04       0  5027.5     .12       0
Bank Sta=4972.5,5027.5
XS Rating Curve= 0 ,0
Exp/Cntr=0.3,0.1

Type RM Length L Ch R = 1 ,134882  ,500,500,500
BEGIN DESCRIPTION:
Willow Creek 20.0
END DESCRIPTION:
XS GIS Cut Line= 3
      2421589.99       829847.61      2423491.67         830147.
      2424779.86       829976.66
#Sta/Elev= 30
  3074.9   87.54  3285.1   77.97  3336.2   72.06  3726.7      58  3888.3   58.06
  4134.1   53.61  4209.6   49.53  4933.6   50.68  4955.1   48.15  4972.5   36.78
    4973   33.45    5027   33.45  5027.5   36.78  5041.3   40.54  5054.8    38.3
  5091.4    41.4  5206.9   36.78  5429.1   39.03    5461   37.33  5501.4   38.49
  5578.8   37.16  5612.7   38.08  5628.2   40.57    5672   39.61  5809.4   41.51
  5966.8   46.18  6046.9   54.62  6113.6   71.23  6224.9   86.06  6299.4   90.98
#Mann= 3 ,0,0
  3074.9     .12       0  4972.5     .04       0  5027.5     .12       0
Bank Sta=4972.5,5027.5
XS Rating Curve= 0 ,0
Exp/Cntr=0.3,0.1

Type RM Length L Ch R = 1 ,134382  ,400,400,400
BEGIN DESCRIPTION:
Willow Creek 19.0
END DESCRIPTION:
XS GIS Cut Line= 3
       2421363.8       831993.65       2423618.5       830525.26
      2424873.31        830131.3
#Sta/Elev= 30
  2309.3   78.96    2914   56.68  3050.4   48.89  3061.4   51.28  3563.2      49
    3579   47.03  3593.8   50.02  3607.5   46.77    3649   49.67  4265.9   49.53
  4438.5   42.78  4535.7   41.09  4618.4   43.15  4683.7   38.86  4721.2   40.35
    4761   38.03  4972.5   36.29    4973   33.22    5027   33.22  5027.5   36.29
    5052   39.19  5287.6   36.79  5494.4   40.31  5528.2   37.06    5584   39.05
    5673   37.87  5727.1   43.69  5970.1   49.64  6114.6   72.06  6315.2   93.09
#Mann= 3 ,0,0
  2309.3     .12       0  4972.5     .04       0  5027.5     .12       0
Bank Sta=4972.5,5027.5
XS Rating Curve= 0 ,0
Exp/Cntr=0.3,0.1

Type RM Length L Ch R = 1 ,133982  ,1000,1000,1000
BEGIN DESCRIPTION:
Willow Creek 18.0
END DESCRIPTION:
XS GIS Cut Line= 3
      2421339.33       832507.24      2423881.01       830786.63
      2424958.87       830202.23
#Sta/Elev= 30
  1930.7   80.26  1965.9   76.04  1974.3   77.66  2410.5   59.43  2550.8   54.72
  2830.6   49.23  3145.3   49.91  3151.7   47.58  3153.4   50.15  3163.6   48.66
    3219      50  3237.6   46.94  3251.4   50.29  3283.5   48.62  3438.4   48.19
  3891.5   50.58  4452.5    48.5  4790.4   41.06  4837.8   43.45  4966.6   41.39
  4970.2   36.24  4970.7    32.8  5029.3    32.8  5029.8   36.24  5479.1   36.62
  5732.2   43.53    5785   55.74  5865.6   77.87  6115.3   92.04  6226.1   93.86
#Mann= 3 ,0,0
  1930.7     .12       0  4970.2     .04       0  5029.8     .12       0
Bank Sta=4970.2,5029.8
XS Rating Curve= 0 ,0
Exp/Cntr=0.3,0.1

Type RM Length L Ch R = 1 ,132982  ,500.9,500.9,500.9
BEGIN DESCRIPTION:
Willow Creek 16.0
END DESCRIPTION:
XS GIS Cut Line= 3
      2422965.66       834367.16      2424668.89       831222.94
      2424922.17       830594.78
#Sta/Elev= 30
  1424.1   82.76  1511.4      80    1754    61.5  1921.6   54.81  2307.9   51.74
  2330.9   48.57  2345.4   52.83  2345.9   50.95  2412.3   48.49  2889.8   47.48
  2905.2   49.54  2927.7   46.76  2982.2   46.31  2990.8   48.62  3205.3   49.53
  3717.4   48.44  4031.8   43.66  4208.1   45.67  4269.2   43.11    4546   42.78
  4588.1   39.78    4715   43.51  4913.6   40.52  4970.2   35.14  4970.7   32.63
  5029.3   32.63  5029.8   35.14  5364.4   38.01    5452   59.68  5677.3   82.01
#Mann= 3 ,0,0
  1424.1     .12       0  4970.2     .04       0  5029.8     .12       0
Bank Sta=4970.2,5029.8
XS Rating Curve= 0 ,0
Exp/Cntr=0.3,0.1

Type RM Length L Ch R = 1 ,132481  ,349.9,349.9,349.9
BEGIN DESCRIPTION:
Willow Creek 15.0
END DESCRIPTION:
XS GIS Cut Line= 3
      2423913.37       834373.21      2425106.34       831255.78
      2425093.37       830594.71
#Sta/Elev= 30
2.31E-11   72.85   173.2   71.03   201.3   65.98   289.1   66.07   457.7   58.53
   770.4   53.06   914.4   48.41  1146.3   48.34  1238.1   45.71  1250.8   47.06
  1339.5   47.46  1792.6   44.26  2020.7   46.32  2094.8   44.02  2354.7   43.84
  2483.1    40.5    2576   42.92  2867.6   41.11  2902.7   42.43  3300.3  36.285
  3339.7   33.44  3373.736.95745  3469.6   38.74  3538.5      38    3591   40.31
  3643.5   50.09  3722.3   53.45  3807.6   63.51  3912.6   79.09  3999.1   85.58
#Mann= 3 ,0,0
2.31E-11     .12       0  3300.3     .04       0  3373.7     .12       0
Bank Sta=3300.3,3373.7
XS Rating Curve= 0 ,0
Exp/Cntr=0.5,0.3

Type RM Length L Ch R = 1 ,132132  ,157.4,157.4,157.4
XS GIS Cut Line= 6
2424368.72477113 833869.458369092424565.91144344833634.789289292
 2424668.7174029 833445.409890292424749.88000247833188.394991645
2425550.68431825830826.5633440922425488.85582631830432.388653409
#Sta/Elev= 30
       0   54.95  280.12   48.94   964.9   47.43 1021.25   44.17 1297.47   44.79
 1695.86   40.85 1737.88   42.21 1799.79   40.02 1841.36   41.81 1893.11   39.23
 1924.51   41.58  2080.4   40.98 2153.15   43.14 2232.83    43.2 2306.06    40.2
 2364.96    43.2 2522.98   37.03 2646.15   35.64 2669.87   32.14 2692.96   35.86
 2708.05   36.23 2715.84   41.41 3040.46   40.84 3137.52   45.42 3305.88   47.27
 3375.62   54.97 3428.75   70.15  3468.6   76.39 3604.76   87.04 3684.42   88.33
#Mann= 3 ,0,0
       0     .12       0 2646.15     .04       0 2692.96     .12       0
#XS Ineff= 2 , 0
       0  2493.8      43  2778.8       0   43.11
Permanent Ineff=
       F       F
Bank Sta=2646.15,2692.96
XS Rating Curve= 0 ,0
Exp/Cntr(USF)=0,0
Exp/Cntr=0.5,0.3

Type RM Length L Ch R = 3 ,132026  ,,,
Node Name=N River Rd Bridg
Bridge Culvert-0,0,0,0, 0
Deck Dist Width WeirC Skew NumUp NumDn MinLoCord MaxHiCord MaxSubmerge Is_Ogee
75,27.5,2.6,0, 65, 65, , , 0.98, 0, 2,2,,
       0   103.6     209   318.1     433   546.4   641.8   753.6   843.5   954.3
  1068.6  1183.8  1233.8  1283.8  1333.8  1383.8  1433.8  1483.8  1533.8  1583.8
  1633.8  1683.8  1733.8  1783.8  1833.8  1883.8  1933.8  1983.8  2033.8  2083.8
  2133.8  2183.8  2233.8  2283.8  2333.8  2383.8  2433.8  2483.8  2533.8  2568.8
  2568.8  2703.8  2703.8  2733.8  2783.8  2833.8  2883.8  2933.8  2983.8  3033.8
  3083.8  3133.8  3183.8  3233.8  3283.8  3333.8  3383.8  3433.8  3483.8  3533.8
  3583.8  3633.8  3683.8  3733.8  3783.8
   56.76   54.48   52.62   52.06   50.95   50.18   49.74   49.18   48.67   47.88
   47.01   46.87   46.45   46.14   45.86    45.6   45.36   45.09    44.8   44.46
   44.22      44   43.79   43.67   43.67   43.57   43.56   43.45   43.38   43.27
   43.24   43.17   43.16   43.07   43.02      43   43.07   43.16   43.25   43.27
   43.27   43.41   43.41   43.19   43.11   43.15   43.29   43.44   43.54   43.83
   44.28   44.83   45.56   46.53   47.44   48.19   48.98   49.89   50.72    51.4
   52.09   52.79   53.52   54.27   55.07
                                                                                
                                                                                
                                                                                
                                                                                
   42.32   42.32
                                                                                
                                        
   -58.1    45.5   150.9     260   374.9   488.3   583.7   695.5   785.4   896.2
  1010.5  1125.7  1175.7  1225.7  1275.7  1325.7  1375.7  1425.7  1475.7  1525.7
  1575.7  1625.7  1675.7  1725.7  1775.7  1825.7  1875.7  1925.7  1975.7  2025.7
  2075.7  2125.7  2175.7  2225.7  2275.7  2325.7  2375.7  2425.7  2475.7  2510.7
  2510.7  2645.7  2645.7  2675.7  2725.7  2775.7  2825.7  2875.7  2925.7  2975.7
  3025.7  3075.7  3125.7  3175.7  3225.7  3275.7  3325.7  3375.7  3425.7  3475.7
  3525.7  3575.7  3625.7  3675.7  3725.7
   56.76   54.48   52.62   52.06   50.95   50.18   49.74   49.18   48.67   47.88
   47.01   46.87   46.45   46.14   45.86    45.6   45.36   45.09    44.8   44.46
   44.22      44   43.79   43.67   43.67   43.57   43.56   43.45   43.38   43.27
   43.24   43.17   43.16   43.07   43.02      43   43.07   43.16   43.25   43.27
   43.27   43.41   43.41   43.19   43.11   43.15   43.29   43.44   43.54   43.83
   44.28   44.83   45.56   46.53   47.44   48.19   48.98   49.89   50.72    51.4
   52.09   52.79   53.52   54.27   55.07
                                                                                
                                                                                
                                                                                
                                                                                
   42.32   42.32
                                                                                
                                        
Pier Skew, UpSta & Num, DnSta & Num=  ,2583.8, 2 ,2525.7, 2 , 0 , 0 , 0 ,,
       1       1
       0      43
       1       1
       0      43
Pier Skew, UpSta & Num, DnSta & Num=  ,2598.8, 2 ,2540.7, 2 , 0 , 0 , 0 ,,
       1       1
       0      43
       1       1
       0      43
Pier Skew, UpSta & Num, DnSta & Num=  ,2613.8, 2 ,2555.7, 2 , 0 , 0 , 0 ,,
       1       1
       0      43
       1       1
       0      43
Pier Skew, UpSta & Num, DnSta & Num=  ,2628.8, 2 ,2570.7, 2 , 0 , 0 , 0 ,,
       1       1
       0      43
       1       1
       0      43
Pier Skew, UpSta & Num, DnSta & Num=  ,2643.8, 2 ,2585.7, 2 , 0 , 0 , 0 ,,
       1       1
       0      43
       1       1
       0      43
Pier Skew, UpSta & Num, DnSta & Num=  ,2658.8, 2 ,2600.7, 2 , 0 , 0 , 0 ,,
       1       1
       0      43
       1       1
       0      43
Pier Skew, UpSta & Num, DnSta & Num=  ,2673.8, 2 ,2615.7, 2 , 0 , 0 , 0 ,,
       1       1
       0      43
       1       1
       0      43
Pier Skew, UpSta & Num, DnSta & Num=  ,2688.8, 2 ,2630.7, 2 , 0 , 0 , 0 ,,
       1       1
       0      43
       1       1
       0      43
Abutment Skew #Up #Dn= , 2 , 2
  2568.8  2588.8
   42.32   32.32
  2510.7  2530.7
   42.32   32.32
BR Coef=-1 , 1 , 1 ,0.9, 0 ,,,0.8,0,1.2,0,
WSPro=,,,, 1 ,,,, 0 ,,,, 0 ,,,,-1 ,-1 ,-1 , 0 , 0 , 0 , 0 , 0
BC Design=,, 0 ,, 0 ,,,,,,
BC Use User HTab Curves=0
BC User HTab FreeFlow(D)= 0

Type RM Length L Ch R = 1 ,131974  ,518.9,518.9,518.9
XS GIS Cut Line= 6
2424514.94662153833929.0353752692424745.31457716833649.314219956
2425022.04600041832826.335992493 2425233.3983525 832144.83248984
2425653.22751447830862.3406662832425570.65001851830402.641947818
#Sta/Elev= 30
       0   55.45  191.47   52.57  234.09   54.08  450.75   49.15 1480.32   44.29
  1645.2   41.56 1731.07   42.24 1775.73    40.3  1923.9   39.99 2038.69   43.81
 2072.15    42.8 2090.81   37.75 2103.07   41.26 2168.06   42.88 2331.16   40.03
 2455.44   40.46 2589.01   36.66 2597.42   32.46  2613.2   30.97 2634.73   31.68
 2640.51   36.69 2672.12   36.87 2714.39   40.51 2971.89   41.03 3400.49   48.85
 3437.16      53 3490.49   70.54 3533.83   76.27 3663.83   86.16 3760.67   86.34
#Mann= 3 ,0,0
       0     .12       0 2589.01     .04       0 2640.51     .12       0
#XS Ineff= 2 , 0
       0 2483.25      43 2673.15       0   43.11
Permanent Ineff=
       F       F
Bank Sta=2589.01,2640.51
XS Rating Curve= 0 ,0
Exp/Cntr(USF)=0,0
Exp/Cntr=0.5,0.3

Type RM Length L Ch R = 1 ,131455  ,466.1,466.1,466.1
BEGIN DESCRIPTION:
Willow Creek 13.0
END DESCRIPTION:
XS GIS Cut Line= 6
      2426105.63       834202.082425700.13048348831171.133791298
2425692.07772532831122.0969287092425707.68311684830977.293063577
2425836.14085427830662.5621628142425552.78964724830084.451245311
#Sta/Elev= 30
       0   76.11   278.1   73.48  615.73   62.29  910.32   57.53    1003   52.03
 1174.76   47.69  1330.7   48.03 1761.01   41.34 2033.41   43.49 2244.28   40.73
    2397   43.65  2655.2   37.82 2985.45   39.13  3060.1  36.831 3080.39   30.33
  3089.5   33.31  3098.6  40.586  3188.1   39.68  3244.2   43.27 3399.03   41.85
 3590.29   47.72 3653.33   53.19  3680.3   52.44 3699.81   57.26 3736.34   58.22
 3817.61   68.84 4003.07   77.13 4061.53   81.08  4182.1   94.66 4237.04   95.41
#Mann= 3 ,0,0
       0     .12       0  3060.1     .04       0  3098.6     .12       0
Bank Sta=3060.1,3098.6
XS Rating Curve= 0 ,0
Exp/Cntr=0.3,0.1

Type RM Length L Ch R = 1 ,130989  ,249.4,249.4,249.4
BEGIN DESCRIPTION:
Willow Creek 12.0
END DESCRIPTION:
XS GIS Cut Line= 4
      2426317.86       834195.75      2426069.81       831041.98
      2425981.62       830917.46      2425649.36       830020.42
#Sta/Elev= 30
       0   75.87   254.1    75.2   507.5   70.82     932   60.17   948.5    56.5
  1014.3   56.41  1201.9   47.57  1600.1   47.14  1725.2   41.04  1985.2   42.24
  2215.6   39.73    2367   42.85    2548   39.47  2656.6    41.6  2923.1      38
  3018.6   40.04 3259.31   38.13  3290.2    34.2  3290.7   31.96  3349.3   31.96
 3355.56   38.19  3435.1   41.45  3529.6   40.44    3687   53.65    3729   53.61
  3753.2   57.56    3806   59.56  4040.4   88.14  4106.9   93.86  4272.7   95.91
#Mann= 3 ,0,0
       0     .12       0 3259.31     .04       0 3355.56     .12       0
Bank Sta=3259.31,3355.56
XS Rating Curve= 0 ,0
Exp/Cntr(USF)=0,0
Exp/Cntr=0.3,0.1

Type RM Length L Ch R = 1 ,130740  ,341.3,341.3,341.3
XS GIS Cut Line= 4
 2426357.1582415833850.2360481852426242.63630005831021.544094523
2426156.74484397830866.9394735742425996.41412595830088.190271756
#Sta/Elev= 30
       0   72.63     502   63.23   520.4   59.74   567.7   58.94   584.1   61.81
   922.4   48.19  1290.1   46.41    1451   40.22    1717   41.94  1835.2   40.14
  2097.9   43.87  2288.3   41.37  2324.5   38.74  2482.1   42.16  2606.9   38.03
  2669.2   39.16  2705.4    36.8  2797.3   39.18  2895.236.92095 2934.37   32.27
  2941.4   32.27  2946.4   36.73  3073.6   40.81  3174.1   38.08    3298   40.72
  3418.6   50.77  3582.7    60.6  3625.5   60.07  3683.2   66.17    3803   72.35
#Mann= 3 ,0,0
       0     .12       0  2895.2     .04       0  2946.4     .12       0
Bank Sta=2895.2,2946.4
XS Rating Curve= 0 ,0
Exp/Cntr(USF)=0,0
Exp/Cntr=0.3,0.1

Type RM Length L Ch R = 1 ,130399  ,309.4,309.4,309.4
XS GIS Cut Line= 3
2426456.58681934833933.4137396882426518.42866772 830990.77245429
2426321.26840336830287.385229145
#Sta/Elev= 30
       0   72.12   240.4    70.4   469.7   65.89   545.6   60.22   798.3   61.36
  1142.8   47.87  1441.5   46.24  1559.3   41.39  1605.5   43.21  1894.3   39.82
  2268.4   43.81  2291.4   42.01  2347.7   42.32  2399.7   40.11  2599.9   40.91
  2675.4   38.55  2724.6   40.36  2968.4   35.66  2995.6   37.98    301637.54132
  3026.7   37.51 3046.96   31.69 3059.31   31.69  3063.8   36.38    307639.26942
  3230.7   42.16  3384.1   47.35    3551   49.12  3632.8   52.01  3673.8   55.62
#Mann= 3 ,0,0
       0     .12       0    3016     .04       0    3076     .12       0
Bank Sta=3016,3076
XS Rating Curve= 0 ,0
Exp/Cntr(USF)=0,0
Exp/Cntr=0.3,0.1

Type RM Length L Ch R = 1 ,130089  ,500,500,500
BEGIN DESCRIPTION:
Willow Creek 10.0
END DESCRIPTION:
XS GIS Cut Line= 3
      2426564.18       834326.21      2426795.53       830867.24
      2427022.73       829855.33
#Sta/Elev= 30
  1533.3    76.1  1904.7   70.71  2265.7   68.89  2279.4   65.76  2327.9   64.27
  3316.1   46.18  3412.3   46.95  3567.9    41.6  3751.7   43.05    3886   41.49
  3930.6   43.77  4050.6   41.26  4232.7   45.26  4486.3   41.92  4509.1   39.68
  4589.5   43.03  4651.9   37.17  4885.6    37.6  4970.2   34.03  4970.7   31.56
  5029.3   31.56  5029.8   34.03  5044.8   40.43  5127.4   40.86  5190.2   38.27
  5274.4   39.59  5416.1   66.76  5639.1   72.48  5700.8   76.92  6037.1   84.29
#Mann= 3 ,0,0
  1533.3     .12       0  4970.2     .04       0  5029.8     .12       0
Bank Sta=4970.2,5029.8
XS Rating Curve= 0 ,0
Exp/Cntr=0.3,0.1

Type RM Length L Ch R = 1 ,129589  ,500,500,500
BEGIN DESCRIPTION:
Willow Creek 9.0
END DESCRIPTION:
XS GIS Cut Line= 3
        2426803.       834135.21      2427261.87       831001.63
      2427395.31       829645.18
#Sta/Elev= 30
    1833   68.64  2167.3   67.01  2176.4   64.42  3244.4   52.81  3462.5   46.93
  3677.4   47.48  3898.4   43.08  4023.7   45.87  4331.5   39.92  4443.4   42.86
  4596.5   39.37  4721.4   42.58  4954.3   38.44  4966.6   36.94  4970.2   33.85
  4970.7   30.89  5029.3   30.89  5029.8   33.85  5058.7   38.92  5284.3   36.37
  5353.2   38.82  5393.1   42.02  5442.9    54.1  5476.9   57.79    5537    57.7
  5551.5   54.05  5563.6   58.55  5627.9   67.63  5810.3   76.67    6363   86.42
#Mann= 3 ,0,0
    1833     .12       0  4970.2     .04       0  5029.8     .12       0
Bank Sta=4970.2,5029.8
XS Rating Curve= 0 ,0
Exp/Cntr=0.3,0.1

Type RM Length L Ch R = 1 ,129089  ,600,600,600
BEGIN DESCRIPTION:
Willow Creek 8.0
END DESCRIPTION:
XS GIS Cut Line= 3
      2427701.01       832597.13      2427680.88       830744.64
      2427643.69       829855.32
#Sta/Elev= 30
  3147.4   55.81  3478.2    52.3  3534.6   48.99  3696.4   45.66  3760.9   47.91
  3874.4   46.75  3948.8   42.85  4042.4   41.27  4488.8   41.89  4541.4   40.07
  4571.2   35.89  4870.8   39.74  4925.5   38.62  4941.9   40.37  4970.2   33.59
  4970.7   30.85  5029.3   30.85  5029.8   33.59    5113    38.4  5184.1   38.47
  5196.6   42.48  5232.5   48.07  5299.5   68.48  5351.2   75.63  5486.1   79.35
  5587.8   68.85  5597.5   63.35  5621.5   69.28    5763   83.05  5890.1   84.86
#Mann= 3 ,0,0
  3147.4     .12       0  4970.2     .04       0  5029.8     .12       0
Bank Sta=4970.2,5029.8
XS Rating Curve= 0 ,0
Exp/Cntr=0.3,0.1

Type RM Length L Ch R = 1 ,128489  ,500,500,500
BEGIN DESCRIPTION:
Willow Creek 7.0
END DESCRIPTION:
XS GIS Cut Line= 3
      2428025.82       832568.46      2427978.38       831059.31
      2428312.41        830008.2
#Sta/Elev= 30
  3490.1   55.59  3989.6   55.85  4069.6   53.75  4197.8   47.07  4370.5   46.88
  4656.5   39.77  4789.3   41.98  4940.9   39.78  4951.8   39.25  4968.8   35.19
  4970.2   33.27  4970.7   30.67  5029.3   30.67  5029.8   33.27  5052.2   37.56
  5069.9   34.41  5113.7   34.48  5150.1   36.01    5179   39.19  5262.4   40.86
  5395.1   37.14  5453.2   39.56  5548.8   39.25  5590.9   42.04  5633.1   50.23
    5678   63.59    5728   74.33    5804   76.77  5970.5   75.25  6102.9   78.73
#Mann= 3 ,0,0
  3490.1     .12       0  4970.2     .04       0  5029.8     .12       0
Bank Sta=4970.2,5029.8
XS Rating Curve= 0 ,0
Exp/Cntr=0.3,0.1

Type RM Length L Ch R = 1 ,127989  ,500,500,500
BEGIN DESCRIPTION:
Willow Creek 6.0
END DESCRIPTION:
XS GIS Cut Line= 3
      2428302.87       832348.67      2428452.55        831112.1
      2428541.69        830189.7
#Sta/Elev= 30
  3754.4   53.22  3876.9   49.72  3929.6   45.01  4035.3   44.43  4145.7    48.7
  4369.7   47.09  4462.8   40.61    4537   43.23  4599.4   42.66  4841.2    36.3
  4909.6   39.72  4921.1   38.79  4935.3   34.37  4970.2   32.95  4970.7   30.83
  5029.3   30.83  5029.8   32.95  5036.3   39.08  5042.7   39.69  5228.2   36.47
  5406.3   38.55  5414.7   36.29  5475.4   37.15  5535.6   41.56  5588.4   47.26
  5617.2   52.69    5702   60.49    5776    60.4  5868.7   69.64  5926.7   70.83
#Mann= 3 ,0,0
  3754.4     .12       0  4970.2     .04       0  5029.8     .12       0
Bank Sta=4970.2,5029.8
XS Rating Curve= 0 ,0
Exp/Cntr=0.3,0.1

Type RM Length L Ch R = 1 ,127489  ,500,500,500
BEGIN DESCRIPTION:
Willow Creek 5.0
END DESCRIPTION:
XS GIS Cut Line= 3
      2428704.09       832482.48      2428881.46       831355.66
      2428761.41       830084.62
#Sta/Elev= 30
  3859.3    50.6  4290.7   50.91  4444.6   45.12  4515.4   39.16  4577.6   38.27
  4654.2   41.21  4766.7   38.17  4825.7   33.94  4879.9   37.92  4933.9   32.85
  4970.2   32.79  4970.7   30.74  5029.3   30.74  5029.8   32.79  5045.8   37.01
  5107.3   39.48  5154.3   36.99  5283.8   35.33  5318.6   36.88  5360.5   34.72
  5401.3    37.3  5460.4   35.99  5533.8   38.97    5557   37.33  5644.5   38.67
  5925.8   35.79    6053   50.27  6094.9   62.87  6168.6   75.75  6276.7   75.81
#Mann= 3 ,0,0
  3859.3     .12       0  4970.2     .04       0  5029.8     .12       0
Bank Sta=4970.2,5029.8
XS Rating Curve= 0 ,0
Exp/Cntr=0.3,0.1

Type RM Length L Ch R = 1 ,126989  ,1500,1500,1500
BEGIN DESCRIPTION:
Willow Creek 4.0
END DESCRIPTION:
XS GIS Cut Line= 4
      2429067.12       832597.09      2429289.27       831610.39
      2429133.99       831221.44      2428971.58       829979.52
#Sta/Elev= 30
  3988.6   52.23  4214.6   45.22  4366.1   43.35  4678.7   44.27  4773.2   37.15
  4951.7   39.82  4964.6   39.14  4970.2   32.47  4970.7   30.47  5029.3   30.47
  5029.8   32.47  5037.6   36.74  5067.6   38.13  5191.7   37.19  5295.4   33.07
  5418.8   37.25  5512.5   37.41  5530.2   33.79  5551.7   32.97  5589.3   35.35
  5679.4   32.75  5727.3   37.14  6076.6   35.14  6207.1      37  6387.2   45.45
  6446.2   51.09  6518.5    62.1  6541.2   68.37  6572.6   73.21  6671.3   76.36
#Mann= 3 ,0,0
  3988.6     .12       0  4970.2     .04       0  5029.8     .12       0
Bank Sta=4970.2,5029.8
XS Rating Curve= 0 ,0
Exp/Cntr=0.3,0.1

Type RM Length L Ch R = 1 ,125489  ,433.1,433.1,433.1
BEGIN DESCRIPTION:
Willow Creek 3.0
END DESCRIPTION:
XS GIS Cut Line= 5
      2429143.55       832625.73      2429563.88       831488.93
      2429563.88       831116.36       2429488.9        830860.3
      2429258.18       829626.08
#Sta/Elev= 30
  3148.6   52.85  3329.4   50.94  3532.1   43.51  3903.6   39.52  3956.5   37.29
  4047.7   39.47  4112.6   37.25  4523.4   38.33  4589.2   35.77  4620.1    37.5
  4780.1   35.45  4790.7    37.1  4814.9   34.91  4938.2   37.07  4970.2   32.33
  4970.7   29.46  5029.3   29.46  5029.8   32.33  5032.5   37.11  5036.3   38.15
  5076.1   40.39  5257.4   39.68  5346.6    36.8  5747.1    51.1  5825.5   51.94
  5924.1   55.72    5943   59.49  6000.3   60.53  6156.8   73.26  6255.6   77.66
#Mann= 3 ,0,0
  3148.6     .12       0  4970.2     .04       0  5029.8     .12       0
Bank Sta=4970.2,5029.8
XS Rating Curve= 0 ,0
Exp/Cntr=0.3,0.1

Type RM Length L Ch R = 1 ,125056  ,166.9,166.9,166.9
XS GIS Cut Line= 6
2429190.79031156832583.4218665282429664.05054148831602.392848248
2429765.11131975831129.1326183242429787.29539302 830914.68657664
 2429713.3484821830443.8912437462429341.14903044829620.615635441
#Sta/Elev= 30
       0   52.17   172.4   50.59   448.8   39.25   591.3   40.74   841.4   37.15
  1030.2   39.09  1117.1   33.84  1184.2   33.24  1335.1   36.19  1479.4   33.68
  1516.3   35.91  1600.334.92726 1618.83   29.43 1645.42   29.43  1658.934.15485
  1678.9   36.84  1728.3   34.12  1797.7   37.68    1967   39.72  2083.3   36.55
  2399.3   42.97  2546.8   40.63  2706.7   46.41  2773.7   46.28  2789.7   48.78
  2824.1    47.5  2849.3   48.71    2977   68.01  3086.9   74.99  3168.8    76.6
#Mann= 3 ,0,0
       0     .12       0  1600.3     .04       0  1658.9     .12       0
Bank Sta=1600.3,1658.9
XS Rating Curve= 0 ,0
Exp/Cntr(USF)=0,0
Exp/Cntr=0.3,0.1

Type RM Length L Ch R = 1 ,124889  ,1646.8,1646.8,1646.8
BEGIN DESCRIPTION:
Willow Creek 2.0
END DESCRIPTION:
XS GIS Cut Line= 5
      2429214.73       832599.32      2429778.59       831766.97
      2429932.49       831112.58      2429892.69       830437.94
      2429395.96       829572.01
#Sta/Elev= 30
  3322.4   52.66  3563.2   50.91  3625.4   48.66  3701.3    39.2  4099.9   37.57
    4350   41.54  4518.6   37.23  4629.2   38.56  4659.9   32.76  4687.5   32.42
  4825.4   35.78  4930.9   35.35  4940.2   32.23  4968.4   34.62  4970.7   29.16
  5029.3   29.16  5030.2   33.54  5102.6    35.1  5137.7   32.01  5192.6   38.74
  5250.4    35.3  5276.5   37.86  5337.3   34.76  5402.9   38.57  5527.9   35.98
  5741.3   42.59  6052.7   40.32  6303.7    46.3  6496.8   70.37  6674.1   75.29
#Mann= 3 ,0,0
  3322.4     .12       0  4968.4     .04       0  5030.2     .12       0
Bank Sta=4968.4,5030.2
XS Rating Curve= 0 ,0
Exp/Cntr=0.3,0.1

Type RM Length L Ch R = 1 ,123242  ,1035.6,1035.6,1035.6
XS GIS Cut Line= 4
2429187.26835221832914.6639122492430559.31162766832012.238860159
 2430646.5863887831110.3996626892429925.56276898829362.770477731
#Sta/Elev= 30
       0   52.32  234.52    51.1  347.57   45.01  382.91   39.28  799.16   40.59
  939.03   34.32 1046.53   32.971877.012   33.95 1900.56      30 1958.61      30
1972.512  34.269 2061.56   32.66 2176.92   33.29 2199.99   35.28 2219.77   33.06
 2460.39   34.58 2523.02   32.86 2907.93   33.04 2950.52   38.47  3014.4   36.82
 3100.09   39.95 3280.99   40.84 3670.99   37.94 4068.48   44.51 4196.25    44.3
 4277.88    46.1 4302.72   57.01 4320.47   62.14 4381.47   72.27 4438.79   76.67
#Mann= 3 ,0,0
       0     .12       01877.012     .04       01972.512     .12       0
Bank Sta=1877.012,1972.512
XS Rating Curve= 0 ,0
Exp/Cntr(USF)=0,0
Exp/Cntr=0.3,0.1

Type RM Length L Ch R = 1 ,122207  ,1211.7,1211.7,1211.7
XS GIS Cut Line= 5
2435312.36128393833477.2585842372431913.68662314832005.760760993
2431634.34353795 831593.397159042431088.95941924831340.658177198
2430211.02400863829292.142219111
#Sta/Elev= 30
       0   75.22  678.08   74.02  881.96   70.98 1321.77   74.31 1357.46   72.57
 1486.44   54.41 1571.97   49.12  3230.4   46.26 3801.69   47.723997.749   37.71
4104.249   37.934144.349   32.914539.249   33.194546.439 30.08344584.329 30.0834
4587.679   33.225297.149   32.945329.049   34.965411.349   32.915464.949   33.54
5497.049   39.335675.549   36.285743.349   39.075861.249   35.035968.249   39.08
6293.049   37.166885.649   42.72 6912.19    46.8 6997.42   68.56 7031.44   72.81
#Mann= 3 ,0,0
       0     .12       04539.249     .04       04587.679     .12       0
Bank Sta=4539.249,4587.679
XS Rating Curve= 0 ,0
Exp/Cntr(USF)=0,0
Exp/Cntr=0.3,0.1

Type RM Length L Ch R = 1 ,120995  ,1445,1445,1445
XS GIS Cut Line= 6
 2435355.9972737833294.8036266032433431.92857639832181.005265482
2432645.29946532831154.4294537362432086.61329493 830462.72276659
2431235.28198767830276.4940431272430344.04452539828587.133480289
#Sta/Elev= 30
       0   75.11  298.86   73.63  683.02   66.25 1005.08   74.01 1243.39   74.87
 1304.04    71.1  1424.2   52.71 1512.54   48.97 1871.52   50.98 2301.69   47.09
 2988.17   53.12 3261.11   47.88  3852.9   48.85  4000.5   38.36  4161.3    40.2
  4276.2   33.08  4396.9      38  4621.3   32.75  4735.5   33.83 4753.18 29.7959
  4799.3 29.7959  4826.2   33.81  5526.3   32.67  5663.5   35.51  5815.9   33.11
    6116   38.63  6702.1   37.03 7055.85   46.78 7152.21   63.54 7187.15   66.41
#Mann= 3 ,0,0
       0     .12       0  4735.5     .04       0  4826.2     .12       0
Bank Sta=4735.5,4826.2
XS Rating Curve= 0 ,0
Exp/Cntr(USF)=0,0
Exp/Cntr=0.3,0.1

Type RM Length L Ch R = 1 ,119550  ,1206.7,1206.7,1206.7
XS GIS Cut Line= 5
2435538.14796616832592.5061144892432871.43434381830795.274058487
2432073.31124325829864.1304411752431860.47841644828893.080668835
2430862.82454075827842.218586439
#Sta/Elev= 30
       0   76.21  429.32   72.92  569.44   68.06  680.52   54.54  959.33   48.13
 1683.49      50 2233.43   47.23  2308.6   49.89 2652.81   47.19 2692.37   43.98
 2826.13   48.013326.803   48.963467.703   38.193644.803   40.963822.903   34.31
4107.203   36.844226.203   32.834628.503   35.164796.503   32.384981.203   35.13
5017.103 29.58765056.353 29.58765058.343   32.455085.303   34.646099.003   37.36
6433.803   43.07 6546.49   70.96 6711.27   81.16 6825.62   71.47  6885.3   86.26
#Mann= 3 ,0,0
       0     .12       04981.203     .04       05085.303     .12       0
Bank Sta=4981.203,5085.303
XS Rating Curve= 0 ,0
Exp/Cntr(USF)=0,0
Exp/Cntr=0.3,0.1

Type RM Length L Ch R = 1 ,118343  ,2589.9,2589.9,2589.9
XS GIS Cut Line= 4
2435812.38400235832123.4404415352433908.99437453829292.142219111
2432791.62203375828786.6642554282431195.37583264827496.365242866
#Sta/Elev= 30
       0   75.78  165.24   74.85  435.75   65.64  705.45   64.05  831.96    58.8
  970.32   63.47 1254.96   59.72 1381.47   62.16 1563.32   52.99 1729.47   52.03
 1824.24   46.66 3566.27   48.594062.223   45.544142.523   39.594281.423   36.31
4628.523   37.464676.423   32.354805.303   33.254824.503 29.16664863.233 29.1666
4870.423   32.615483.823    35.85794.323   33.526005.223   38.756199.323    34.7
6397.123      446490.423   61.06 6559.06   58.69 6626.56   78.45 6690.54   87.56
#Mann= 3 ,0,0
       0     .12       04805.303     .04       04870.423     .12       0
Bank Sta=4805.303,4870.423
XS Rating Curve= 0 ,0
Exp/Cntr(USF)=0,0
Exp/Cntr=0.3,0.1

Type RM Length L Ch R = 1 ,115753  ,806.6,806.6,806.6
XS GIS Cut Line= 5
 2436296.1571335831177.3789987612433736.06770274828201.373981688
2433070.96511895827123.9077959412432525.58100023826817.960607396
2431554.53122789826551.919573878
#Sta/Elev= 30
       0   76.87  327.19   73.51 1034.71   73.88 1164.54   68.55 1207.82   62.59
 1290.34   61.97 1497.39   52.79 1518.33   55.23 1627.75    51.9 1679.54   47.25
 3592.41   45.83  3886.6   48.03 4072.16   43.024259.745   42.814456.345   36.78
4706.145   39.754926.045   33.955099.645      375403.445   32.355501.245   33.51
5542.115 28.55195595.945 28.55195629.635   33.656051.945   32.076426.145   38.68
6507.745   41.61 6559.73   49.64  6692.4   60.42 6791.05   64.73 6824.03   63.37
#Mann= 3 ,0,0
       0     .12       05501.245     .04       05629.635     .12       0
Bank Sta=5501.245,5629.635
XS Rating Curve= 0 ,0
Exp/Cntr(USF)=0,0
Exp/Cntr=0.3,0.1

Type RM Length L Ch R = 1 ,114947  ,2646.4,2646.4,2646.4
XS GIS Cut Line= 6
2436506.86475571830327.0078165012435665.68101097828662.947260791
2435012.16395629827121.7016839362433855.78616782826392.294953767
2433031.05896392826232.6703336572431754.06200303826192.764178629
#Sta/Elev= 30
       0   73.82  448.11   69.47  631.92   65.18   650.3   61.22     665   63.61
 1127.33   50.09 1902.68    48.9  2066.6   45.61 2444.34   48.47  3075.1   43.88
 3762.64   46.75 3844.48   44.77  3917.8   37.48 3999.26   36.16 4569.47    39.9
 4740.14   33.06 5565.97   32.93 5582.58    28.5 5650.54    28.5 5665.72  32.739
 6547.57   32.47 6580.39   34.57 6629.63    63.3 6649.32   71.09 6698.96    72.2
 6731.79   87.54 6761.33   78.27 6781.02   76.25 6938.58   80.93 7023.52   79.16
#Mann= 3 ,0,0
       0     .12       0 5565.97     .04       0 5665.72     .12       0
Bank Sta=5565.97,5665.72
XS Rating Curve= 0 ,0
Exp/Cntr(USF)=0,0
Exp/Cntr=0.3,0.1

Type RM Length L Ch R = 1 ,112301  ,928.9,928.9,928.9
XS GIS Cut Line= 6
2436845.25404783830162.3137287622435824.70917647828453.030082329
2435185.09062807826810.0825230542433070.96511895825740.494421649
2432911.34049883825168.506199586 2432412.0305175825028.867346813
#Sta/Elev= 30
       0   74.82  468.83    71.8  717.21   60.38 1076.39   52.69 1615.17   51.58
 1779.48   46.43 2622.51   44.96 3070.59   47.98  3454.5   44.34 3852.74   47.58
 4000.32   46.87 4131.93   36.73 4195.19   35.53 4724.66   37.93 5092.34   31.19
 5351.37   34.62 5452.67   31.84  5717.4   32.13 6088.75   36.38 6352.69    31.8
 6379.44   28.22 6438.28   28.37 6452.69    31.8  6860.7   33.11 6881.14   37.72
 6918.61   53.82 6924.31   58.99 6968.59    66.4 7115.08   73.65 7235.44   70.94
#Mann= 3 ,0,0
       0     .12       0 6352.69     .04       0 6452.69     .12       0
Bank Sta=6352.69,6452.69
XS Rating Curve= 0 ,0
Exp/Cntr(USF)=0,0
Exp/Cntr=0.3,0.1

Type RM Length L Ch R = 1 ,111372  ,1367.5,1367.5,1367.5
XS GIS Cut Line= 6
2437023.97630107829773.2855632612435951.93170887828115.890371467
2435351.49027653826580.2337792272433815.88001279825727.192369973
2433762.67180609824889.1631143922433487.74094491824370.135094029
#Sta/Elev= 30
       0   76.03  153.07   75.09  500.61   60.11  739.35   58.23  906.97   53.27
 1051.54   57.36 1090.62   54.44 1421.97   53.09 1562.42   46.14 1699.84   48.73
  1719.7   46.02 1965.77   45.41 2302.05   47.53  2935.4   45.25 3055.17   47.72
 3442.67   44.69 3562.44   46.87  3823.3   43.95 4003.44   35.38 4442.55   40.56
 4639.92   30.87 5976.97   31.81 6001.29   27.75 6063.36   27.75 6076.03   31.78
 6398.37   34.85 6495.48   56.87 6580.87   59.65 6721.96   75.48 6806.46   78.39
#Mann= 3 ,0,0
       0     .12       0 5976.97     .04       0 6076.03     .12       0
Bank Sta=5976.97,6076.03
XS Rating Curve= 0 ,0
Exp/Cntr(USF)=0,0
Exp/Cntr=0.3,0.1

Type RM Length L Ch R = 1 ,110004  ,806.9,806.9,806.9
XS GIS Cut Line= 6
2437244.55996009829557.6742970612436098.23762113827867.806433285
2435438.27996358826428.2392384542435159.38723206825328.130819696
 2434973.1585086824729.5384942812434599.89166701823522.315303443
#Sta/Elev= 30
       0   72.67  243.37   74.19  360.17   69.66  429.97   63.06   681.6   57.23
 1270.22   57.96 1417.98   51.13 1440.69   47.98 1733.57   43.78 2436.57   48.24
  3508.5   46.65  3732.4   42.16 3905.02   45.84 3959.84   44.86 4044.46   34.48
 4389.69   35.53    4454   30.47 5092.81  30.042 5102.83    27.2 5189.36  27.188
 5193.31   30.17  5589.9   30.09 5672.31   33.67  5892.1   30.03 5936.74   34.71
 6211.47   35.67 6283.58   41.73 6372.27   67.51 6410.65   73.58 6651.03    78.1
#Mann= 3 ,0,0
       0     .12       0 5092.81     .04       0 5193.31     .12       0
Bank Sta=5092.81,5193.31
XS Rating Curve= 0 ,0
Exp/Cntr(USF)=0,0
Exp/Cntr=0.3,0.1

Type RM Length L Ch R = 1 ,109197  ,627.6,627.6,627.6
XS GIS Cut Line= 6
2437302.31201948829283.1254347552436496.23123741827657.880528999
2435917.60417759825940.0251967872435824.48981585825288.224664669
2435877.69802256824543.3097708192435455.99423927823058.701601788
#Sta/Elev= 30
       0   75.81  258.99   70.23   383.5   62.74  573.94   57.33 1141.58   58.39
 1272.85   45.66 1701.26   42.99  2505.3   47.74 2950.87   42.91 3780.33   48.43
 3859.87   42.54 3942.73   31.51 4606.48  29.932 4624.06      27 4693.98   26.99
 4706.48  30.744 5044.05    29.9  5156.6   33.93 5241.87   29.79 5398.76   29.66
  5477.2   32.59 5900.12   31.81 6114.99   36.92 6237.77   35.91 6333.72   40.59
 6353.73   44.56 6358.89   48.87 6427.11   72.34 6471.44   80.61 6575.42   83.85
#Mann= 3 ,0,0
       0     .12       0 4606.48     .04       0 4706.48     .12       0
Bank Sta=4606.48,4706.48
XS Rating Curve= 0 ,0
Exp/Cntr(USF)=0,0
Exp/Cntr=0.3,0.1

Type RM Length L Ch R = 1 ,108570  ,740.5,740.5,740.5
XS GIS Cut Line= 3
2437667.08948707829172.4274730882436409.78008959826006.535455167
2436383.17598624822800.741001277
#Sta/Elev= 30
       0   74.27  155.12   74.09  334.51   68.49  441.18   61.02  483.46   64.49
  776.54   55.41 1224.87    58.3 1383.72   49.24  1627.3   48.38 1719.08   43.69
 2015.61   42.66 2358.03   47.15 2605.14   43.95 2876.95    48.4 3285.65   48.25
3576.025   45.033717.025   32.673825.325   29.914205.925   30.124232.555 26.8471
4261.225 26.84714265.025   29.915231.925   29.675318.125   34.485482.225   35.57
5629.825   30.785948.125    35.26446.825   34.216532.125   38.34 6612.33      58
#Mann= 3 ,0,0
       0     .12       04205.925     .04       04265.025     .12       0
Bank Sta=4205.925,4265.025
XS Rating Curve= 0 ,0
Exp/Cntr(USF)=0,0
Exp/Cntr=0.3,0.1

Type RM Length L Ch R = 1 ,107829  ,1220.7,1220.7,1220.7
XS GIS Cut Line= 6
2438799.50307077827886.5290338732437540.45448204826232.670333657
2437167.99703512825368.0369747242436888.65394993824011.227703783
2436976.38923923823010.8500332872436831.97988289822329.092522954
#Sta/Elev= 30
       0    75.4  393.09   73.98  453.72   73.08  482.58   69.75  499.07   73.13
  635.15   70.91  864.31   56.48  999.72   51.28 2405.93   44.16 2441.79   42.39
 2523.95   30.06 2902.79   31.28 3044.38    29.5 3084.57   31.63 3185.97  29.489
 3205.97  26.671 3271.14  26.671 3285.97  30.081 4022.47   29.47 4102.86   34.24
  4233.5   30.76 4354.09   35.61 4483.51   31.99  4793.1   30.75 5630.16   35.73
 5717.36   40.09 5794.93   57.34 5888.83   70.59 5942.49   74.09 6106.38   78.02
#Mann= 3 ,0,0
       0     .12       0 3185.97     .04       0 3285.97     .12       0
Bank Sta=3185.97,3285.97
XS Rating Curve= 0 ,0
Exp/Cntr(USF)=0,0
Exp/Cntr=0.3,0.1

Type RM Length L Ch R = 1 ,106608  ,1317.6,1317.6,1317.6
XS GIS Cut Line= 5
2439277.80066999827554.5290338732439003.68016639 825900.11904176
2437966.12013567824543.3097708192437625.28530067822766.641838121
2436938.44195263822297.469149598
#Sta/Elev= 30
       0   74.86  468.45   73.87  498.31   70.28  544.87   69.72  661.26   58.61
  923.98   52.03  1472.7   49.19  1602.4   45.77 2129.54   49.12 2278.91   43.62
 2318.94   29.61 2335.46    31.7 2592.16   30.44 2613.77    32.9 2694.78   29.44
 3030.89   29.35 3050.89  26.382 3115.87  26.382 3121.49   29.29  3692.9   29.43
 3760.68   33.12 4551.45   31.08  4604.9   33.77  4999.1   33.12 5593.96   38.24
 5622.89   40.83 5705.33   60.39 5776.85   72.28 5856.31   76.62 6025.88   76.77
#Mann= 3 ,0,0
       0     .12       0 3030.89     .04       0 3121.49     .12       0
Bank Sta=3030.89,3121.49
XS Rating Curve= 0 ,0
Exp/Cntr(USF)=0,0
Exp/Cntr=0.3,0.1

Type RM Length L Ch R = 1 ,105291  ,822.4,822.4,822.4
XS GIS Cut Line= 5
2440587.97627018 826738.104410742440067.84430046 824929.06926942
2439176.60683818824157.5502722182438644.52477114823425.937430044
 2438164.2985646821695.083468513
#Sta/Elev= 30
       0   73.33  235.54   71.08  372.09   60.35  477.91   55.27   747.6   47.11
 1355.25   49.27 1662.49   47.04 2126.04   47.72 2164.37   46.86 2289.77   33.68
 2595.46   29.54 2801.82   31.82  2846.1   29.24 3479.42   31.34 3510.35 26.0689
 3564.96 26.0689 3580.78   31.17 4047.84   29.24 4210.98   33.38 4313.41   31.77
 4473.44   33.86 4657.29    30.4 4895.63   33.17 5413.15   33.97 5484.65   38.74
 5509.64   43.33 5577.73   61.77 5632.21   70.02 5673.07   74.15 5761.99   77.52
#Mann= 3 ,0,0
       0     .12       0 3479.42     .04       0 3580.78     .12       0
Bank Sta=3479.42,3580.78
XS Rating Curve= 0 ,0
Exp/Cntr(USF)=0,0
Exp/Cntr=0.3,0.1

Type RM Length L Ch R = 1 ,104468  ,1462.6,1462.6,1462.6
XS GIS Cut Line= 5
2442208.31740435825459.9814291142440679.73867755824835.954907688
2439655.48069851823931.4153937282439655.48069851823000.271776416
2438977.07606304821231.098903522
#Sta/Elev= 30
       0    70.6  469.83   73.84  551.33   70.23  685.99   56.21  778.13   51.35
  941.14   47.12 1136.04   47.67 1323.86   44.84 2013.96   48.14 2164.48   46.58
2200.252   45.062287.452   30.042314.152   29.192471.352   32.412536.952   29.38
3392.852   30.183403.982 25.87383450.592 25.87383454.452   30.144336.252   29.57
4515.652   31.284789.752   29.274940.852   35.675120.052    31.85204.352   37.07
5462.552   37.42 5606.15   54.35 5658.86   54.47 5739.67    49.4 5843.47   49.63
#Mann= 3 ,0,0
       0     .12       03392.852     .04       03454.452     .12       0
Bank Sta=3392.852,3454.452
XS Rating Curve= 0 ,0
Exp/Cntr(USF)=0,0
Exp/Cntr=0.3,0.1
