HEC-RAS study MapleSwamp.prj: S-26-65 over Maple Swamp

--- MapleSwamp.g04 (geometry) --- (continued)

Type RM Length L Ch R = 1 ,22251   ,420.4,420.4,420.4
BEGIN DESCRIPTION:
Maple Swamp 34.0
END DESCRIPTION:
XS GIS Cut Line= 3
      2609877.57       770461.53      2608843.86       769958.05
      2607840.06       769544.65
#Sta/Elev= 30
  3850.2   39.88  3894.4   39.46  3946.1   36.05  4005.2   35.31  4116.9   32.02
  4214.6   27.24    4348   28.52  4388.1   28.08  4414.8   28.88  4581.6   27.72
  4612.5   26.78  4926.6   27.58    4983   26.65    4984   24.65    5016   24.65
    5017   26.65  5021.1   27.29  5047.4   26.65  5174.1   27.74  5242.1   26.78
  5371.9   28.17  5404.3   27.47  5591.3   28.17  5631.4   27.25  5706.2    28.1
  5730.2   27.28  5798.1   29.65  5826.1   33.19  5867.1   35.95  6085.6   39.74
#Mann= 3 ,-1,0
  3850.2     .15       0    4983     .05       0    5017     .15       0
Bank Sta=4983,5017
XS Rating Curve= 0 ,0
Exp/Cntr=0.3,0.1

Type RM Length L Ch R = 1 ,21830   ,613.8,613.8,613.8
BEGIN DESCRIPTION:
Maple Swamp 33.0
END DESCRIPTION:
XS GIS Cut Line= 3
      2610349.39       769544.66      2608960.33        769555.1
      2607818.64       769464.24
#Sta/Elev= 30
  3610.9   45.41  3660.3   44.79  3720.3   43.13  3766.1    40.9  3853.8   38.85
  4098.6    34.7  4230.3   28.78  4290.3   27.76  4377.6   27.02  4650.3   27.79
  4717.3   27.17  4747.1   27.74  4950.3   27.18    4983   26.51    4984   24.51
    5016   24.51    5017   26.51  5040.5   27.15  5423.2   26.74  5461.8   27.44
  5491.9   26.65  5702.5   28.21  5732.6    27.4  5762.7   27.75  5822.9   33.64
    5853   35.37    5925   35.01  5964.8   36.26  6003.5   38.83  6145.3   41.72
#Mann= 3 ,-1,0
  3610.9     .15       0    4983     .05       0    5017     .15       0
Bank Sta=4983,5017
XS Rating Curve= 0 ,0
Exp/Cntr=0.3,0.1

Type RM Length L Ch R = 1 ,21216   ,529.6,529.6,529.6
BEGIN DESCRIPTION:
Maple Swamp 32.0
END DESCRIPTION:
XS GIS Cut Line= 3
      2610209.99       768962.93      2609054.98       768948.78
      2607915.18       769011.18
#Sta/Elev= 30
  3844.9   39.59  3907.1   37.09  4174.4    32.5  4234.9   32.98  4264.9   34.26
  4324.9   34.04  4410.9   32.11  4474.9   26.83  4504.9   26.47  4692.4    26.3
    4775   26.79  4825.9   26.29    4955   27.24    4983   26.25    4984   24.25
    5016   24.25    5017   26.25  5225.3   26.73  5255.4   27.57  5285.4   26.25
  5435.6   26.81  5480.8   26.37  5537.6   26.77    5676   26.53    5706   27.93
  5766.1   33.76  5796.2   35.16  5862.2   35.69  6006.5   40.52  6141.5   43.59
#Mann= 3 ,-1,0
  3844.9     .15       0    4983     .05       0    5017     .15       0
Bank Sta=4983,5017
XS Rating Curve= 0 ,0
Exp/Cntr=0.3,0.1

Type RM Length L Ch R = 1 ,20687   ,518.6,518.6,518.6
BEGIN DESCRIPTION:
Maple Swamp 31.0
END DESCRIPTION:
XS GIS Cut Line= 3
      2610314.77       768618.94      2609104.15       768421.65
      2608250.25       768363.13
#Sta/Elev= 30
  3773.4   43.66    3910   38.13  4008.2   36.16  4122.7    34.3    4221   34.89
  4273.2   34.59  4335.5   33.44  4363.8   31.39  4426.7   29.44  4457.1   26.35
  4487.5   25.85  4717.5   26.35  4822.1   27.52  4882.6   26.37  4978.9   26.02
  4981.6   25.23  4982.6   23.23  5017.4   23.23  5018.4   25.23  5124.4   25.67
  5174.3   26.84  5230.6   26.59  5286.9   27.27    5365   26.55    5470   26.78
  5484.5   26.74  5568.3   32.77  5652.7   35.88  5818.9   39.17  5855.9   39.18
#Mann= 4 ,-1,0
  3773.4     .15       0  4981.6     .05       0  5018.4     .15       0
    5470      .1       0
Bank Sta=4981.6,5018.4
XS Rating Curve= 0 ,0
Exp/Cntr=0.3,0.1

Type RM Length L Ch R = 1 ,20168   ,627.7,627.7,627.7
BEGIN DESCRIPTION:
Maple Swamp 30.0
END DESCRIPTION:
XS GIS Cut Line= 3
      2610033.01       767799.45      2609031.18       767916.14
      2608190.56       768035.16
#Sta/Elev= 30
  3991.4   39.22  4070.2   36.55  4182.8   34.39  4326.7   26.01  4356.9   26.43
  4417.3    25.4    4450   25.85  4477.7   25.09  4628.7   25.13  4658.9   25.75
  4689.1   25.45  4779.7   26.27  4840.1   24.74  4960.9   25.08  4981.6   24.56
  4982.6   22.56  5017.4   22.56  5018.4   24.56  5172.5   25.65  5278.7   24.68
    5385   25.92  5448.1   25.57  5464.5   26.11  5506.2      31  5536.5   32.62
  5566.8    35.3  5644.5   38.46  5748.6   38.82  5778.9   38.26    5849   38.29
#Mann= 3 ,-1,0
  3991.4     .15       0  4981.6     .05       0  5018.4     .15       0
Bank Sta=4981.6,5018.4
XS Rating Curve= 0 ,0
Exp/Cntr=0.3,0.1

Type RM Length L Ch R = 1 ,19541   ,430.6,430.6,430.6
BEGIN DESCRIPTION:
Maple Swamp 29.0
END DESCRIPTION:
XS GIS Cut Line= 3
      2609684.52       767157.12      2608713.26       767376.83
      2608049.17       767655.77
#Sta/Elev= 30
  4004.2   39.49  4142.1   36.89  4234.4   34.33  4265.2    31.7  4326.7   25.38
  4417.1   24.55  4695.4    25.3  4757.3   24.49  4849.6   24.51  4973.6   25.41
  4981.6   24.49  4982.6   22.49  5017.4   22.49  5018.4   24.49  5018.9    25.1
  5036.1   25.29  5133.7   24.85  5157.7    25.9  5198.8   26.33  5231.3   27.29
  5263.8   27.06  5296.4   27.52    5360   30.66  5386.8   31.84  5432.6   32.46
  5459.1   33.73    5616   34.29  5661.8   36.04  5684.7   35.48  5720.3   36.17
#Mann= 4 ,-1,0
  4004.2     .15       0  4981.6     .05       0  5018.4     .15       0
    5360      .1       0
Bank Sta=4981.6,5018.4
XS Rating Curve= 0 ,0
Exp/Cntr=0.3,0.1

Type RM Length L Ch R = 1 ,19110   ,494.3,494.3,494.3
BEGIN DESCRIPTION:
Maple Swamp 28.0
END DESCRIPTION:
XS GIS Cut Line= 3
      2609604.06       766374.34      2608666.04       766950.23
       2607915.2       767612.83
#Sta/Elev= 30
  3899.3   42.24  3977.3   42.09  4033.1   40.02  4160.8   37.95    4174    36.9
  4228.8   35.55  4368.8   29.88  4400.8   28.21  4426.2   25.44  4455.6   24.75
  4770.2   24.29  4807.6   25.21  4981.6   24.03  4982.6   22.03  5017.4   22.03
  5018.4   24.03    5045   25.11  5101.4   25.54    5453   24.84  5501.5    25.6
    5570   27.71  5581.6   28.74    5615   29.18  5691.3   31.32  5755.1   32.45
  5781.6   32.19  5815.8   34.67  5925.1    35.9  5981.7   38.63  6001.4   38.13
#Mann= 4 ,-1,0
  3899.3     .15       0  4981.6     .05       0  5018.4     .15       0
    5615      .1       0
Bank Sta=4981.6,5018.4
XS Rating Curve= 0 ,0
Exp/Cntr=0.3,0.1

Type RM Length L Ch R = 1 ,18616   ,512.9,512.9,512.9
BEGIN DESCRIPTION:
Maple Swamp 27.0
END DESCRIPTION:
XS GIS Cut Line= 3
      2609164.39       766133.07      2608439.67       766522.45
       2607362.9       767537.82
#Sta/Elev= 30
  4177.3   36.73  4318.5   34.67  4445.5   34.74  4556.9    38.8    4591   38.85
  4650.9    34.9    4699   27.74  4727.2   24.65  4897.5   23.61  4952.6   24.23
  4981.6   23.61  4982.6   21.61  5017.4   21.61  5018.4   23.61  5040.8   24.37
    5082   23.62  5111.2   24.49  5196.1   25.17  5259.8   24.76    5281   25.44
  5491.1   25.05  5579.5    27.4  5710.7   25.71  5896.4   24.78  5947.9   27.22
  6016.8   28.35  6071.6   30.96  6112.9   35.47  6195.3   39.38    6480   39.45
#Mann= 3 ,-1,0
  4177.3     .15       0  4981.6     .05       0  5018.4     .15       0
Bank Sta=4981.6,5018.4
XS Rating Curve= 0 ,0
Exp/Cntr=0.3,0.1

Type RM Length L Ch R = 1 ,18103   ,474.6,474.6,474.6
BEGIN DESCRIPTION:
Maple Swamp 26.0
END DESCRIPTION:
XS GIS Cut Line= 3
      2608364.58       765723.91      2608034.62       766217.12
      2607352.17        767221.5
#Sta/Elev= 30
  4406.6   40.46    4438   40.39  4510.2    37.2    4544   36.64  4585.5   31.75
  4657.5   33.41  4723.6   29.95  4798.9   23.76    4835   23.44  4907.2    24.4
  4981.6   23.14  4982.6   21.14  5017.4   21.14  5018.4   23.14  5019.8   23.89
  5051.8   23.41  5106.6   24.55    5171   23.54  5233.2   25.05  5322.1    24.2
  5414.5   24.58  5450.8   24.06  5506.4   26.07  5595.9   26.32    5741    24.2
  5933.5   23.75  6013.2   25.38  6103.7   32.87  6139.9   34.64  6214.3   35.46
#Mann= 3 ,-1,0
  4406.6     .15       0  4981.6     .05       0  5018.4     .15       0
Bank Sta=4981.6,5018.4
XS Rating Curve= 0 ,0
Exp/Cntr=0.3,0.1

Type RM Length L Ch R = 1 ,17628   ,381.7,381.7,381.7
BEGIN DESCRIPTION:
Maple Swamp 25.0
END DESCRIPTION:
XS GIS Cut Line= 3
       2608033.1       765473.06      2607626.74       765986.51
       2607041.2       767044.03
#Sta/Elev= 30
  4345.2   38.19  4380.8   37.65  4468.8   38.14    4509   37.43    4573   31.16
  4698.4   31.24  4831.3   26.73  4875.9   24.33  4954.1   24.24  4981.6   23.47
  4982.6   21.47  5017.4   21.47  5018.4   23.47  5055.2   23.47  5117.1   25.12
  5198.8   25.06  5220.9   24.56  5353.3   25.49  5375.4    24.8  5484.1   25.12
  5555.1   24.64  5618.2   23.72  5689.8   24.31  5828.8    23.5  5895.6   24.24
  5984.2   24.42  6015.4   25.11    6056   28.01  6135.6   32.06  6208.8    35.2
#Mann= 3 ,-1,0
  4345.2     .15       0  4981.6     .05       0  5018.4     .15       0
Bank Sta=4981.6,5018.4
XS Rating Curve= 0 ,0
Exp/Cntr=0.3,0.1

Type RM Length L Ch R = 1 ,17246   ,305.8,305.8,305.8
BEGIN DESCRIPTION:
Maple Swamp 24.0
END DESCRIPTION:
XS GIS Cut Line= 3
      2607834.74       765306.82      2607363.54       765712.08
      2606354.95        766550.7
#Sta/Elev= 30
  4378.5   38.03  4460.1   38.95  4518.8   38.67  4561.4   33.54  4603.9   30.03
  4747.6   24.44  4774.1   25.69  4816.7   22.64  4880.5   23.69  4981.6   22.43
  4982.6   20.43  5017.4   20.43  5018.4   22.43  5199.7   25.47  5221.2   24.17
  5293.9   23.61  5575.5   23.92  5628.9   25.15  5669.3   24.68  5721.1   25.99
  5761.3   25.18    5863   24.86  5997.8   25.65  6073.3   24.74    6123    25.4
  6152.3   27.31  6185.5   30.81  6214.1   32.48  6279.3    39.3  6311.7   41.15
#Mann= 3 ,-1,0
  4378.5     .15       0  4981.6     .05       0  5018.4     .15       0
Bank Sta=4981.6,5018.4
XS Rating Curve= 0 ,0
Exp/Cntr=0.3,0.1

Type RM Length L Ch R = 1 ,16941   ,381.2,381.2,381.2
XS GIS Cut Line= 6
2607663.03915865765162.1287914282607317.86565341765380.157168759
2607188.07094694765462.3635095792607183.85640032765464.959821024
2606400.84357699766318.1206746062606231.62611154766502.444958671
#Sta/Elev= 30
  4432.9   37.25  4472.1   36.71  4578.6   37.72  4643.9   35.98  4720.5   29.15
  4730.9   27.45  4791.5   24.55  4861.3      23  4981.6   22.55  4982.6   20.55
  5017.4   20.55  5018.4   22.55  5020.3   24.37    5061   24.33  5101.7   22.77
  5183.1   23.34  5227.1   24.83  5316.1   23.85  5468.2   23.76    5544   26.22
  5607.7   24.86  5735.1   25.32  5804.2   26.42  5875.4   25.21  5981.6   25.81
  6119.7   25.11  6244.7   31.57  6287.2    35.9  6350.9   40.21  6408.1   41.55
#Mann= 3 ,-1,0
  4432.9     .15       0  4981.6     .05       0  5018.4     .15       0
Bank Sta=4981.6,5018.4
XS Rating Curve= 0 ,0
Exp/Cntr(USF)=0,0
Exp/Cntr=0.3,0.1

Type RM Length L Ch R = 1 ,16560   ,651.5,651.5,651.5
BEGIN DESCRIPTION:
Maple Swamp 22.0
END DESCRIPTION:
XS GIS Cut Line= 3
      2607310.11       764724.83      2606896.75       765215.26
      2606046.31       766223.49
#Sta/Elev= 30
  4358.6   34.37  4467.4   37.03  4539.8   36.54  4582.3   35.68  4646.2   31.64
  4667.5   29.56  4795.8   26.61  4859.1   22.31  4953.9   23.21  4981.6   22.31
  4982.6   20.31  5017.4   20.31  5018.4   22.31    5026   23.25  5071.6   23.94
  5242.3   22.52  5305.2   22.84  5327.5   24.02  5370.5   24.55  5464.1   23.55
  5582.7   24.97  5646.8   23.87  5723.9   25.86  5770.4   23.33  5817.2   25.25
    5857   25.83    5910   24.48  6013.5   24.78  6093.9   26.21    6319   34.24
#Mann= 3 ,-1,0
  4358.6     .15       0  4981.6     .05       0  5018.4     .15       0
Bank Sta=4981.6,5018.4
XS Rating Curve= 0 ,0
Exp/Cntr=0.3,0.1

Type RM Length L Ch R = 1 ,15908   ,551.1,551.1,551.1
BEGIN DESCRIPTION:
Maple Swamp 21.0
END DESCRIPTION:
XS GIS Cut Line= 3
      2606691.25       764329.67      2606353.35       764861.62
      2605994.11       766245.87
#Sta/Elev= 30
  4369.8   38.68  4488.7   38.34  4666.4   33.62    4697   31.97  4762.2   23.09
    4773   22.69  4808.5   21.93    4936   21.49  4979.5   22.48  4981.5   21.49
  4982.5   19.49  5017.5   19.49  5018.5   21.49  5048.9   22.52  5235.9   22.02
  5297.9   22.31  5328.9   23.44  5390.3   23.67  5483.9   22.79  5542.8   23.87
  5641.2   23.25  5700.8   25.47  5731.8   25.56  5788.9   23.42  5862.7   24.16
  6034.9   24.32  6165.8   28.32  6196.8   28.45  6351.7   32.94  6430.1   34.16
#Mann= 3 ,-1,0
  4369.8     .15       0  4981.5     .05       0  5018.5     .15       0
Bank Sta=4981.5,5018.5
XS Rating Curve= 0 ,0
Exp/Cntr=0.3,0.1

Type RM Length L Ch R = 1 ,15357   ,373.7,373.7,373.7
BEGIN DESCRIPTION:
Maple Swamp 20.0
END DESCRIPTION:
XS GIS Cut Line= 3
      2606594.28        764313.3       2605915.6       764671.07
      2605013.64       765230.37
#Sta/Elev= 30
  4232.8   37.83  4550.7   34.21  4588.1   32.69    4622   29.27  4685.1   23.94
  4757.6   22.65  4796.1   22.34  4825.5   22.76  4927.2   21.63  4961.1   22.17
  4981.5   21.45 5090.88    21.8 5097.73   19.07 5115.33   19.07 5120.35   21.83
    5136   21.99  5170.3   21.19  5206.6   21.64  5241.9   21.22  5301.1   21.29
  5588.4   22.72  5671.5    26.4  5681.1   27.39  5700.8   28.59    5733   30.02
  5794.9   32.61  5851.9   34.04  5912.6   36.33  5983.2   37.72  6061.3   37.47
#Mann= 3 ,0,0
  4232.8     .15       0 5090.88     .05       0 5120.35     .15       0
Bank Sta=5090.88,5120.35
XS Rating Curve= 0 ,0
Exp/Cntr=0.5,0.3

Type RM Length L Ch R = 1 ,14983   ,178.4,178.4,178.4
BEGIN DESCRIPTION:
Maple Swamp (HWY-65) US
END DESCRIPTION:
XS GIS Cut Line= 6
2606270.99543383 764294.697914162606020.25670458764349.151248127
2605826.05042104764407.279025191      2605492.18         764527.
2605378.51949651764553.548940603 2604612.5311043 764655.20192812
#Sta/Elev= 30
       0   34.78  160.37    33.9  194.95      32  218.45   33.68  265.63   29.41
  279.33   29.34  295.24   25.84  300.58   23.26  466.37   21.34  470.14    18.8
  510.62    18.8     515    21.1  562.23   22.96  653.45   21.53  705.54   21.97
  715.93   23.06  760.97   21.54  826.44   21.39  973.91   23.36 1013.62   22.54
 1155.94   22.85 1165.86   23.88 1195.65   24.12 1318.11   22.59 1397.54   22.93
 1483.59   26.03 1496.83   28.94 1549.78   33.77 1661.85   40.97 1703.46   42.18
#Mann= 3 ,0,0
       0     .15       0  466.37     .05       0     515     .15       0
#XS Ineff= 2 , 0
         377.495   28.54 603.875           28.69
Permanent Ineff=
       F       F
Bank Sta=466.37,515
XS Rating Curve= 0 ,0
Exp/Cntr=0.5,0.3

Type RM Length L Ch R = 3 ,14910   ,,,
BEGIN DESCRIPTION:
Maple Swamp (HWY-65) TOR
Structure ID: LDS_MPS_02
Approximate Survey Structure
END DESCRIPTION:
Bridge Culvert--1,0,-1,-1, 0
Deck Dist Width WeirC Skew NumUp NumDn MinLoCord MaxHiCord MaxSubmerge Is_Ogee
60.69,27.5,3,0, 18, 17, , , 0.95, 0, 2,2,,
  14.185  67.655 235.905 341.185 438.185 438.185 543.185 543.185 642.285 944.585
1073.6851173.3851273.5851373.7851473.7851573.9851668.5851733.385
   34.25    33.2   30.36   28.54      29      29      29      29   28.69   29.28
   29.02   28.93   29.08   29.63    30.9    32.5      34   34.85
                                           27.77   27.77
                                                                
       0  143.48  341.73     447     544     544     649     649   748.1  1050.4
  1149.5  1249.2  1349.4  1449.6  1549.6  1649.8  1719.2
   34.25    33.2   30.36   28.54      29      29      29      29   28.69   29.28
   29.02   28.93   29.08   29.63    30.9    32.5      34
                                           27.77   27.77
                                                        
Pier Skew, UpSta & Num, DnSta & Num=  ,453.185, 2 ,559, 2 , 0 , 0 , 0 ,,
       1       1
   13.99   27.77
       1       1
   13.99   27.77
Pier Skew, UpSta & Num, DnSta & Num=  ,468.185, 2 ,574, 2 , 0 , 0 , 0 ,,
       1       1
   13.99   27.77
       1       1
   13.99   27.77
Pier Skew, UpSta & Num, DnSta & Num=  ,483.185, 2 ,589, 2 , 0 , 0 , 0 ,,
       1       1
   13.99   27.77
       1       1
   13.99   27.77
Pier Skew, UpSta & Num, DnSta & Num=  ,498.185, 2 ,604, 2 , 0 , 0 , 0 ,,
       1       1
   13.99   27.77
       1       1
   13.99   27.77
Pier Skew, UpSta & Num, DnSta & Num=  ,513.185, 2 ,619, 2 , 0 , 0 , 0 ,,
       1       1
   13.99   27.77
       1       1
   13.99   27.77
Pier Skew, UpSta & Num, DnSta & Num=  ,528.185, 2 ,634, 2 , 0 , 0 , 0 ,,
       1       1
   13.99   27.77
       1       1
   13.99   27.77
Abutment Skew #Up #Dn= , 2 , 2
 438.185 458.185
    27.7    17.7
     544     564
    27.7    17.7
Abutment Skew #Up #Dn= , 2 , 2
 523.185 543.185
   17.77   27.77
     629     649
   17.77   27.77
BR Coef=-1 , 1 , 1 ,0.9, 0 ,,,0.8,0,1.2,0,
WSPro=,,,, 1 ,,,, 0 ,,,, 0 ,,,,-1 ,-1 ,-1 , 0 , 0 , 0 , 0 , 0
BC Design=,, 0 ,, 0 ,,6,453.185,559,15,1
BC HTab HWMax=42.97
BC Use User HTab Curves=0
BC User HTab FreeFlow(D)= 0

Type RM Length L Ch R = 1 ,14805   ,280.5,280.5,280.5
BEGIN DESCRIPTION:
Maple Swamp (HWY-65) DS
END DESCRIPTION:
XS GIS Cut Line= 6
2606230.15242302764153.3335826612605956.41891485764221.747375249
2605717.76125913764299.580046683 2605609.6181506764338.869154525
2605425.12236869  764389.45403362604591.13352491764525.198147551
#Sta/Elev= 30
       0   34.19  334.55   32.54  400.54   29.55  431.18   26.79  441.53   22.63
  451.88   21.67  479.49   21.62  496.83   24.56  513.07   25.55  538.37   24.98
  563.19   22.43  575.61    18.7  617.11    18.7  621.84    22.4  696.63   23.34
  850.33   21.66  883.58   24.03  926.51   24.54 1116.29   22.37 1169.63   24.09
 1206.05   22.78 1249.26   25.44 1282.51   23.09 1355.65   22.88 1362.29   24.54
 1378.92   22.72 1425.46   22.94 1481.97   25.24 1491.95   27.63 1684.52   31.84
#Mann= 3 ,0,0
       0     .15       0  563.19     .05       0  621.84     .15       0
#XS Ineff= 2 , 0
         498.895   28.54 694.105           28.69
Permanent Ineff=
       F       F
Bank Sta=563.19,621.84
XS Rating Curve= 0 ,0
Exp/Cntr=0.5,0.3

Type RM Length L Ch R = 1 ,14524   ,509.7,509.7,509.7
BEGIN DESCRIPTION:
Maple Swamp 19.0
END DESCRIPTION:
XS GIS Cut Line= 3
       2606299.2       763639.26      2605460.96       764145.41
      2604377.67       764551.49
#Sta/Elev= 30
       0   41.09   642.6   28.69   673.2   28.57   711.6    22.5   767.1   23.39
     875   21.36   937.7   23.57   960.7   21.49961.9998    18.6996.4001    18.6
   997.7   21.49  1119.9   21.52    1204   24.36  1358.2   22.34  1407.2   23.82
  1487.8   22.79    1508   24.23  1526.4   22.66  1664.1   23.87  1701.6   22.76
  1754.1   23.48  1768.1   25.54  1785.7   28.06  1844.5   26.66  1881.9      30
  1939.8   31.53  2041.4   31.69  2051.9   28.03    2080   31.16  2136.1   33.53
#Mann= 5 ,-1,0
       0      .1       0   642.6     .15       0   960.7    .052       0
   997.7     .15       0  1768.1      .1       0
#XS Ineff= 2 , 0
                         1221.89           28.69
Permanent Ineff=
       F       F
Bank Sta=960.7,997.7
XS Rating Curve= 0 ,0
Exp/Cntr=0.5,0.3

Type RM Length L Ch R = 1 ,14015   ,224,224,224
BEGIN DESCRIPTION:
Maple Swamp 18.0
END DESCRIPTION:
XS GIS Cut Line= 3
      2605946.63       763453.24      2605045.68       763884.86
      2604033.18       764206.97
#Sta/Elev= 30
       0      40   186.3    36.1   345.9   36.34   393.6   37.98   415.1   38.27
   426.4   32.44   440.9   28.62     510   26.99   539.1   27.09   550.9   31.29
     561   30.86   568.2   26.56   571.9   26.56   581.3   21.89   771.2   21.47
   848.4   22.94  988.45   21.31   992.6   18.36 1009.84   18.36 1013.27   21.32
    1139   23.47  1295.7   22.18  1355.7   23.34  1403.9   22.28  1692.7   22.88
  1792.9   27.66  1830.8   28.12    1910   35.73  1951.3   37.75  2061.5   39.42
#Mann= 5 ,-1,0
       0      .1       0   393.6     .08       0     510     .14       0
996.2998    .052       0  1004.7     .15       0
Bank Sta=988.45,1013.27
XS Rating Curve= 0 ,0
Exp/Cntr=0.3,0.1

Type RM Length L Ch R = 1 ,13791   ,437.1,437.1,437.1
BEGIN DESCRIPTION:
Maple Swamp 17.0
END DESCRIPTION:
XS GIS Cut Line= 3
      2605872.17       763450.02      2604962.43        763680.6
      2603742.02       763935.25
#Sta/Elev= 30
       0   39.24   194.6   37.62   269.1   38.84   289.4   40.37   340.2   33.83
   357.1   27.77   455.2   28.31   485.7   26.55   519.5   27.03   529.7   27.28
   537.4   30.46   546.6   30.44   566.9   25.84   573.7   22.63   597.4   21.36
   763.2   22.61   780.2   21.54919.1001   21.37920.3999    18.3956.6001    18.3
957.8999   21.37  1699.6   23.42  1817.3   27.67  1899.2   28.33  1911.2   32.28
  1924.6   34.67  1951.4   34.55  1981.5   38.54  2048.6    42.1  2185.2   42.87
#Mann= 5 ,-1,0
       0      .1       0   289.4     .08       0   519.5     .15       0
919.1001    .052       0957.8999     .15       0
Bank Sta=919.1001,957.8999
XS Rating Curve= 0 ,0
Exp/Cntr=0.3,0.1

Type RM Length L Ch R = 1 ,13354   ,586,586,586
BEGIN DESCRIPTION:
Maple Swamp 16.0
END DESCRIPTION:
XS GIS Cut Line= 3
      2606024.98         763325.      2604987.82       763245.56
      2603688.63       763338.41
#Sta/Elev= 30
       0   42.57     201    42.5   319.4    40.8   339.2   39.57   372.1      35
   395.1   30.94   414.9   30.76     428   25.11   641.9   25.65   655.4   26.04
   681.4   22.62   707.7   22.27  1020.8    21.3  1022.1    18.1  1058.3    18.1
  1059.6    21.3    1165   20.34  1224.2   22.12    1244   20.94  1747.2   22.97
    1790   24.04  1859.1    29.5  1868.9   27.91  1901.8   28.18  1921.6   30.29
  1951.2   29.68  1964.3   33.89  1980.8   35.65  2082.7   39.94  2342.7   44.05
#Mann= 5 ,-1,0
       0      .1       0   372.1     .08       0   641.9     .14       0
  1020.8    .052       0  1059.6     .15       0
Bank Sta=1020.8,1059.6
XS Rating Curve= 0 ,0
Exp/Cntr=0.3,0.1

Type RM Length L Ch R = 1 ,12767   ,675.8,675.8,675.8
BEGIN DESCRIPTION:
Maple Swamp 15.0
END DESCRIPTION:
XS GIS Cut Line= 3
      2606117.24       762986.01      2605078.07       762666.77
      2603879.09       762561.43
#Sta/Elev= 30
       0   40.66   223.8    35.5   254.7   36.01   271.1   35.32   290.9   30.67
     302   29.87   334.1   29.22   357.9   32.69     440   26.28   676.8   20.28
   838.2    20.5   855.3   21.92   865.6   20.84  1067.7   21.21    1069   18.06
  1105.2   18.06  1106.5   21.21  1757.2   21.24  1796.7   22.81  1806.6   24.53
  1832.5   23.65  1869.2   26.46  1882.4   29.85  1914.2   28.28  1941.6   29.04
  1964.7   30.83  1974.6   35.76  2010.5    38.8  2033.9   38.09  2290.7   42.27
#Mann= 3 ,-1,0
       0     .15       0  1067.7    .052       0  1106.5     .15       0
Bank Sta=1067.7,1106.5
XS Rating Curve= 0 ,0
Exp/Cntr=0.3,0.1

Type RM Length L Ch R = 1 ,12092   ,452.6,452.6,452.6
BEGIN DESCRIPTION:
Maple Swamp 14.0
END DESCRIPTION:
XS GIS Cut Line= 3
       2606032.3       761851.79      2605221.51       762006.37
      2604073.23       762130.79
#Sta/Elev= 30
       0   36.24   151.3   37.75   298.3   34.99   385.1   26.21     472   20.31
   522.1   21.73   565.5   20.16   662.3   19.75     806   20.91807.2998   17.45
   843.5   17.45   844.1   20.54  1021.1   22.07  1152.7   19.84  1208.8   20.78
  1235.2    19.6  1393.3   19.86  1443.1   21.74  1515.7    21.1  1614.7   22.72
  1654.3   26.55  1680.7   23.35  1729.8   23.47  1763.2   26.08  1776.4   25.81
  1786.3   29.57  1789.6   29.56  1799.5   38.59  1802.8   40.38  1980.4    41.6
#Mann= 3 ,-1,0
       0     .15       0     806    .052       0844.7998     .15       0
Bank Sta=806,844.1
XS Rating Curve= 0 ,0
Exp/Cntr=0.3,0.1

Type RM Length L Ch R = 1 ,11639   ,595,595,595
BEGIN DESCRIPTION:
Maple Swamp 13.0
END DESCRIPTION:
XS GIS Cut Line= 3
      2606111.14       761572.78      2605307.21       761562.06
      2604309.81       761560.65
#Sta/Elev= 30
       0   40.59   204.6   39.76   358.2   35.89     385   32.67   404.7    31.7
   457.2   26.57   519.5   24.08   542.5   21.32   585.2    19.5   650.8   20.72
   663.9   19.41   686.9   19.91   693.4   20.78   726.3   19.81  784.57   20.14
785.8999    17.2822.1001    17.2  822.79   20.09  1047.8   19.38  1192.1   20.13
  1244.6   19.54  1267.6   20.24  1487.4   19.89  1523.5   20.72  1536.6   21.93
  1569.4   28.51  1615.4   32.49  1690.8   34.61  1759.7   38.24  1801.4   38.85
#Mann= 4 ,-1,0
       0      .1       0     385     .15       0784.6001    .052       0
823.3999     .15       0
Bank Sta=784.57,822.79
XS Rating Curve= 0 ,0
Exp/Cntr=0.3,0.1

Type RM Length L Ch R = 1 ,11044   ,564.8,564.8,564.8
BEGIN DESCRIPTION:
Maple Swamp 12.0
END DESCRIPTION:
XS GIS Cut Line= 3
      2606220.38       760887.39      2605379.14       760972.13
      2604048.95       761178.53
#Sta/Elev= 30
       0   40.41   206.5   39.06   279.1   37.06   387.9   30.12   440.7   23.72
   480.2   22.12   486.8   19.93   529.7   19.57   542.9   21.85   549.5   25.16
   559.4   26.56   569.3   22.38   572.6   22.38   582.5   19.26  826.45   19.27
827.3999    16.8863.6001    16.8  864.43    19.1  1221.4   19.67    1341    18.8
  1440.6   20.44  1520.2   19.35    1663   19.96  1692.9   21.97  1759.5   22.98
  1792.5   25.45    1819    25.9  1858.9   31.53    1922   31.89  2191.6   38.25
#Mann= 3 ,0,0
       0      .1       0  826.45     .05       0  864.43     .15       0
Bank Sta=826.45,864.43
XS Rating Curve= 0 ,0
Exp/Cntr=0.3,0.1

Type RM Length L Ch R = 1 ,10479   ,981.1,981.1,981.1
BEGIN DESCRIPTION:
Maple Swamp 11.0
END DESCRIPTION:
XS GIS Cut Line= 3
      2605989.85       760156.52      2605192.76        760447.1
      2603854.91       760944.99
#Sta/Elev= 30
       0   39.79   287.7    38.8     340   37.22   385.4   34.78   395.9   29.86
   411.4   25.51   451.8   22.88     581   22.84     588      24   612.4   22.84
   710.8   22.85   727.7    23.9   766.1   19.63   825.4   20.24828.7998   19.22
830.1001   16.72866.6997   16.72     868   19.22   870.9   20.41   940.9      19
   989.3   20.44  1072.5   20.34  1204.2   18.33  1476.6    19.9  1511.5   19.12
  1574.5   22.31  1749.5   24.97  1834.4   34.15  2068.1   39.34  2275.9   41.25
#Mann= 5 ,-1,0
       0      .1       0388.3999     .08       0718.3999     .13       0
828.7998    .052       0     868     .15       0
Bank Sta=825.4,870.9
XS Rating Curve= 0 ,0
Exp/Cntr=0.3,0.1

Type RM Length L Ch R = 1 ,9498    ,733.3,733.3,733.3
BEGIN DESCRIPTION:
Maple Swamp 10.0
END DESCRIPTION:
XS GIS Cut Line= 3
      2605322.69       759167.85      2604659.46       759627.79
       2603794.2       760617.49
#Sta/Elev= 30
       0   40.21    67.6   40.44    79.9   38.63    95.9   38.34   115.9   36.36
   151.8   26.24   167.8   22.72   195.7   19.22   219.7   17.73   510.9   18.25
   533.9    17.5   543.1   18.33   666.8    17.9   698.8   19.12   758.6   18.07
   786.6      19   787.5   18.59788.8003   16.09825.3999   16.09826.7002   18.59
   826.9   18.78  1184.3   17.94  1689.8   18.86  1829.2   24.16  1861.4   26.76
  1896.2   31.96  1942.7   35.74  1964.3   35.57  2038.4    38.7  2121.7   40.43
#Mann= 3 ,-1,0
       0      .1       0   787.5     .05       0826.7002     .15       0
Bank Sta=786.6,826.9
XS Rating Curve= 0 ,0
Exp/Cntr=0.3,0.1

Type RM Length L Ch R = 1 ,8765    ,843.9,843.9,843.9
BEGIN DESCRIPTION:
Maple Swamp 9.0
END DESCRIPTION:
XS GIS Cut Line= 3
      2605235.11       759046.19      2604153.55       758839.16
       2603131.1       758661.87
#Sta/Elev= 30
       0   39.25  141.39   38.71  214.51    34.7   224.9   31.56  238.27   28.88
  244.95   28.66  261.65   24.26  291.71      20   315.1   18.84   348.5   17.75
  398.61   18.47  472.09   17.26  571.94   17.72   572.7   15.52   609.7   15.52
  610.54   17.78  936.41    17.7  953.11   18.47 1176.68   17.53 1289.89   17.94
  1313.3   18.89 1393.12   17.82 1628.29   17.78 1729.43   20.68 1739.42   20.12
 1819.33   24.06 1899.25   25.55 2025.78   33.41 2052.42   36.32  2138.9   36.25
#Mann= 3 ,-1,0
       0     .15       0  571.94     .05       0  610.54     .15       0
Bank Sta=571.94,610.54
XS Rating Curve= 0 ,0
Exp/Cntr=0.3,0.1

Type RM Length L Ch R = 1 ,7921    ,1107.5,1107.5,1107.5
BEGIN DESCRIPTION:
Maple Swamp 8.0
END DESCRIPTION:
XS GIS Cut Line= 3
      2605537.84       758379.27       2604163.1       757844.74
      2603235.94       757719.37
#Sta/Elev= 30
       0   35.23    33.8      34    51.4   32.32   89.64   31.98  118.28   29.03
  181.64   28.72  311.88   20.62  421.01   17.19  473.81   17.94  551.28   16.91
  579.41   17.72   697.3   17.41   698.5   14.91   735.5   14.91   736.7   17.41
  832.86   17.93  896.22   16.69 1002.44   16.81 1026.47   17.82 1068.71   17.03
 1389.04   17.88  1434.8      17 1817.92   17.47 2019.88   24.07 2046.36   26.22
 2099.33   27.36  2152.3   31.37 2231.76   35.23 2354.45   38.97  2410.6      39
#Mann= 3 ,-1,0
       0     .15       0   697.3     .05       0   736.7     .15       0
Bank Sta=697.3,736.7
XS Rating Curve= 0 ,0
Exp/Cntr=0.3,0.1

Type RM Length L Ch R = 1 ,6813    ,662,662,662
BEGIN DESCRIPTION:
Maple Swamp 7.0
END DESCRIPTION:
XS GIS Cut Line= 3
      2606256.07       757139.43      2604391.01       756989.26
      2603480.51       756988.03
#Sta/Elev= 30
       0   34.63   232.1   32.05   311.1   25.72  380.22   25.79  482.26   21.29
   505.3   22.45  525.04   21.38  564.54   21.49  627.08   19.24   656.7   17.09
  738.99   16.93  781.78   15.34 1083.83   15.77  1084.6   14.32  1121.6   14.32
 1122.64   15.82 1400.57   15.71 1443.36   16.57 1456.53   15.77 1644.14   15.78
 1726.43    17.5 2166.87   16.92 2317.44   17.72 2379.78   19.57 2432.27   23.69
 2583.19   25.02 2619.28   28.67 2642.25   33.01 2681.27    36.7  2781.6   37.81
#Mann= 3 ,-1,0
       0     .15       0 1083.83     .05       0 1122.64     .15       0
Bank Sta=1083.83,1122.64
XS Rating Curve= 0 ,0
Exp/Cntr=0.3,0.1

Type RM Length L Ch R = 1 ,6151    ,334.1,334.1,334.1
XS GIS Cut Line= 6
2606023.27567147756510.1735210862604834.47600654756334.871384243
2604637.37371215756305.2100602962604627.57540168756304.216163674
2604153.89617531 756275.640474692603542.84476962756238.518487706
#Sta/Elev= 30
       0   30.71   227.4   27.52   247.3   26.38   253.9   24.88   267.2   25.22
   280.4   23.95   340.1   24.57   452.9   17.96   539.1    15.3   675.1   16.41
   698.8    15.3  764.32   15.59  765.37   14.09  803.97   14.09  805.19   15.42
   993.4   15.34  1053.1   16.71  1172.5   15.28  1361.6   17.31  1743.3   16.54
  1759.7   17.97  1795.9   17.18  1864.9   17.74  1927.4   19.62  1976.7   22.53
  2042.4   34.14  2081.8   36.29  2246.2   39.09  2417.1   38.71  2497.5   39.83
#Mann= 3 ,0,0
       0     .15       0  764.32     .05       0  805.19     .15       0
Bank Sta=764.32,805.19
XS Rating Curve= 0 ,0
Exp/Cntr(USF)=0,0
Exp/Cntr=0.5,0.3

Type RM Length L Ch R = 1 ,5817    ,125.9,125.9,125.9
BEGIN DESCRIPTION:
Maple Swamp (Co Jo Rd) US
END DESCRIPTION:
XS GIS Cut Line= 4
2606014.47930916756336.3196717752605489.55930916756092.069671775
2604730.09930916755988.9496717752603699.54930916755889.799671775
#Sta/Elev= 30
       0   30.37   205.8   29.41   245.6   27.45   256.5   25.76   304.9    25.5
   433.8   21.46   460.5      22   531.5   18.24   553.2   18.81   564.1   16.63
   571.3   17.94  747.89   15.13  748.38    14.1  788.01    14.1  788.52   15.14
  1111.4   16.38  1164.6   15.56  1322.7   16.88  1327.9    14.1  1362.9    14.1
  1369.8   16.94    1383   17.31    1406   16.44  1491.7   17.38  1738.9   16.33
  1916.9   17.17  2022.4   19.47  2045.5   22.42  2118.8   25.84  2380.7   27.61
#Mann= 3 ,0,0
       0     .15       0  747.89     .05       0  788.52     .15       0
#XS Ineff= 3 ,-1
       0  668.65   19.51  875.05 1284.55   19.67 1409.55  2380.7      20
Permanent Ineff=
       F       F       F
Bank Sta=747.89,788.52
XS Rating Curve= 0 ,0
Exp/Cntr=0.5,0.3

Type RM Length L Ch R = 4 ,5755    ,,,
BEGIN DESCRIPTION:
Maple Swamp (Co Jo Rd) TOR
Structure ID: Maple Swamp_CJR
Approximate Survey Structure. The top of bridge is curb
END DESCRIPTION:
Bridge Culvert--1,0,-1,-1, 0
Deck Dist Width WeirC Skew NumUp NumDn MinLoCord MaxHiCord MaxSubmerge Is_Ogee
47.23342,28.5,3,0, 50, 50, , , 0.95, 0, 2,2,,
       0    56.2    89.9   134.7   158.1   176.7   201.4   243.7   274.8   304.7
   317.4   355.4   375.9   396.5   445.9   460.3   510.1  715.85  715.85  827.85
  827.85   871.5    1162  1225.1  1284.3  1317.3 1324.55 1324.55 1369.55 1369.55
  1432.8  1455.9  1531.8  1571.4    1611  1657.2  1690.1  1719.8  1772.4  1825.4
  1901.3    1931  1977.1  2006.8  2059.6    2086  2142.6  2214.7  2285.9  6028.9
   29.48   28.22   27.36   26.19   26.01   25.78   25.94   25.66   24.56    24.3
   24.16    24.3   24.82   23.93   21.44   21.38   19.51   20.22   21.02   21.11
   20.31   19.67   19.67   19.78   20.08   20.19   20.19   20.89   20.94   20.24
   20.36   20.38   20.74   20.81   20.96   21.19   21.23    21.4   21.62   21.85
   22.27   22.53   22.82   23.03    23.2   23.41   24.07   24.64   25.66   27.21
                                                                                
                                                                   19.32   19.41
                                                           19.29   19.34
                                                                                
                                                                                
       0    91.2   139.7   184.2   212.9   232.3     254   290.7   329.9     357
   376.2   420.5   442.2   487.9   503.7   555.2   586.3   777.6   777.6   889.6
   889.6   928.1    1209  1250.9  1301.5  1351.1 1370.95 1370.95 1415.95 1415.95
  1467.1    1493    1559  1618.4    1658  1714.1  1737.1  1766.8  1816.3  1855.9
  1918.6  1964.8  2007.8  2040.6  2076.2  2116.5  2172.6  2238.6    2321  2423.3
   29.48   28.22   27.14   26.23   25.84   25.58   25.63   25.66   24.94   24.04
   24.73   24.78   23.96   21.33   21.56   19.51   19.51   20.22   21.02   21.11
   20.31   19.67   19.67   19.58   19.81   20.16   20.19   20.89   20.94   20.24
   20.37   20.46   20.69   20.81   20.96   21.06   21.23    21.4   21.66   21.91
   22.03   22.45   22.78   22.94   22.92   23.31   23.79    24.5   25.53   26.96
                                                                                
                                                                   19.32   19.41
                                                           19.29   19.34
                                                                                
                                                                                
Pier Skew, UpSta & Num, DnSta & Num=  ,729.85, 2 ,791.6, 2 , 0 , 0 , 0 ,,
       1       1
       0      20
       1       1
       0      20
Pier Skew, UpSta & Num, DnSta & Num=  ,743.85, 2 ,805.6, 2 , 0 , 0 , 0 ,,
       1       1
       0      20
       1       1
       0      20
Pier Skew, UpSta & Num, DnSta & Num=  ,757.85, 2 ,819.6, 2 , 0 , 0 , 0 ,,
       1       1
       0      20
       1       1
       0      20
Pier Skew, UpSta & Num, DnSta & Num=  ,771.85, 2 ,833.6, 2 , 0 , 0 , 0 ,,
       1       1
       0      20
       1       1
       0      20
Pier Skew, UpSta & Num, DnSta & Num=  ,785.85, 2 ,847.6, 2 , 0 , 0 , 0 ,,
       1       1
       0      20
       1       1
       0      20
Pier Skew, UpSta & Num, DnSta & Num=  ,799.85, 2 ,861.6, 2 , 0 , 0 , 0 ,,
       1       1
       0      20
       1       1
       0      20
Pier Skew, UpSta & Num, DnSta & Num=  ,813.85, 2 ,875.6, 2 , 0 , 0 , 0 ,,
       1       1
       0      20
       1       1
       0      20
Pier Skew, UpSta & Num, DnSta & Num=  ,1339.55, 2 ,1385.95, 2 , 0 , 0 , 0 ,,
       1       1
       0    28.2
       1       1
       0    28.2
Pier Skew, UpSta & Num, DnSta & Num=  ,1354.55, 2 ,1400.95, 2 , 0 , 0 , 0 ,,
       1       1
       0    28.2
       1       1
       0    28.2
Abutment Skew #Up #Dn= , 2 , 2
  715.85  721.85
   19.32   16.32
   777.6   783.6
   19.32   16.32
Abutment Skew #Up #Dn= , 2 , 2
  821.85  827.85
   16.41   19.41
   883.6   889.6
   16.41   19.41
Abutment Skew #Up #Dn= , 2 , 2
 1324.55 1330.55
   19.29   16.29
 1370.95 1376.95
   19.29   16.29
Abutment Skew #Up #Dn= , 2 , 2
 1363.55 1369.55
   16.34   19.34
 1409.95 1415.95
   16.34   19.34
BR Coef=-1 ,-1 ,-1 ,0.9, 0 ,,,0.8,0,1.2,0,
WSPro=,,,, 1 ,,,, 0 ,,,, 0 ,,,,-1 ,-1 ,-1 , 0 , 0 , 0 , 0 , 0
BC Mult= 3 ,0,1083.7,0,1130.28
BC Mult= 3 ,1083.7,4000,1130.28,4000
BC Design=,, 0 ,, 0 ,,,,,,
BC HTab HWMax=30.34
BC Use User HTab Curves=0
BC User HTab FreeFlow(D)= 0

Type RM Length L Ch R = 1 ,5691    ,180.1,180.1,180.1
BEGIN DESCRIPTION:
Maple Swamp (Co Jo Rd) DS
END DESCRIPTION:
XS GIS Cut Line= 4
2606089.06714504756228.8342747832605516.53714504755962.704274783
2604758.30714504755882.7142747832603723.95714504755764.294274783
#Sta/Elev= 30
       0   30.26   175.9   28.98   345.9   24.84   414.7   25.59   461.7   23.91
   479.8   19.66     516      20   541.3   17.28   595.6   15.35   724.1   17.17
  808.46   15.85  808.93   13.84  849.77   13.84  850.04   15.83  1133.2   15.63
  1255.2   17.25  1367.4   15.99  1376.3   13.84  1411.3   13.84  1416.4   16.25
    1440   16.45  2011.3   16.68  2021.2   17.51  2034.4   21.11    2087   24.54
  2186.3   25.11  2199.5   26.62  2315.1   27.62  2361.4   30.03  2434.9   30.94
#Mann= 3 ,0,0
       0     .15       0  808.46     .05       0  850.04     .15       0
#XS Ineff= 3 ,-1
       0   752.5   19.51   914.7 1349.25   19.58 1437.55  2380.7      20
Permanent Ineff=
       F       F       F
Bank Sta=808.46,850.04
XS Rating Curve= 0 ,0
Exp/Cntr=0.5,0.3

Type RM Length L Ch R = 1 ,5511    ,621.4,621.4,621.4
BEGIN DESCRIPTION:
Maple Swamp 5.0
END DESCRIPTION:
XS GIS Cut Line= 3
      2605968.59       756047.89      2604904.81       755566.09
      2603157.48       755219.89
#Sta/Elev= 30
       0   24.28   60.84   25.42  215.72   24.75  258.93   21.42  288.64   15.66
  670.35   15.52   671.8   13.24   709.8   13.24  710.77   15.42  712.74   15.76
   835.2   14.95  903.63   15.97  964.86   14.73  1091.2    15.9 1287.05   15.22
  1313.8   16.34 1661.64   16.24 1698.43   14.87 1932.56   15.35 1962.66   15.82
 1976.04   18.38 1986.07   16.16 2049.62   17.53 2170.03   22.47 2287.09   24.09
  2467.7   31.59 2578.07   34.42 2705.16   34.09 2818.88   36.18  2949.1   35.74
#Mann= 3 ,-1,0
       0     .15       0  670.35     .05       0  712.74     .15       0
#XS Ineff= 2 , 0
           470.3   19.24  1531.3           19.19
Permanent Ineff=
       F       F
Bank Sta=670.35,712.74
XS Rating Curve= 0 ,0
Exp/Cntr=0.5,0.3

Type RM Length L Ch R = 1 ,4890    ,1193.5,1193.5,1193.5
BEGIN DESCRIPTION:
Maple Swamp 4.0
END DESCRIPTION:
XS GIS Cut Line= 3
      2605978.84       755986.58      2605437.48       755098.47
      2605263.27        754177.2
#Sta/Elev= 30
       0   21.51   25.32   21.85  136.82   19.56  176.61   17.31  186.77   15.58
  195.52   15.31  321.26   15.38  340.47   16.09  378.89   15.03  451.89   14.78
  471.11   15.57  521.06   14.84  555.64   15.94  601.74   15.04  920.41   15.06
   927.8   12.22   965.8   12.22     969   14.78  970.61   14.87 1303.59    15.6
  1330.3   14.55    1347   15.44 1373.71   14.93 1433.81   16.66 1660.86   18.49
 1677.56    19.8 1707.61   18.85 1747.68   19.22 1857.86   22.88  1977.7   23.71
#Mann= 3 ,-1,0
       0     .15       0  920.41     .05       0  970.61     .15       0
Bank Sta=920.41,970.61
XS Rating Curve= 0 ,0
Exp/Cntr=0.3,0.1

Type RM Length L Ch R = 1 ,3696    ,1148.8,1148.8,1148.8
BEGIN DESCRIPTION:
Maple Swamp 3.0
END DESCRIPTION:
XS GIS Cut Line= 3
      2607185.09       755628.79      2606597.15       754772.63
      2605345.06       754146.53
#Sta/Elev= 30
       0   30.91     253   25.38   300.7   26.63   401.7   26.11     436   23.15
   507.9   23.31   579.3   21.72   619.1   19.51     631   17.67   698.7   14.92
   714.6   15.62   734.4   14.63 1018.49   14.55  1019.6   12.32  1057.6   12.32
 1058.64   14.43  1150.4   15.49    1210    14.6  1248.4   15.33  1310.2    14.5
  1634.6   15.22  1733.3   14.32  1781.3   15.39    1814   14.77  1825.3   15.16
  1836.3   17.12  1860.4   19.38  1945.3   21.25  2111.5   22.44  2438.5   22.76
#Mann= 3 ,0,0
       0     .15       0 1018.49     .05       0 1058.64     .15       0
Bank Sta=1018.49,1058.64
XS Rating Curve= 0 ,0
Exp/Cntr=0.3,0.1

Type RM Length L Ch R = 1 ,2548    ,1055.7,1055.7,1055.7
BEGIN DESCRIPTION:
Maple Swamp 2.0
END DESCRIPTION:
XS GIS Cut Line= 3
      2608084.66       755618.55      2607528.73        754104.7
      2606653.54       752786.96
#Sta/Elev= 30
       0   37.95    85.4   34.15   158.8   27.62   264.1   24.98   274.8      26
   331.9   24.94   382.5   25.95   396.5   24.81   501.3   25.69   595.7   23.28
   722.1   23.91  1036.2   20.03  1043.8   19.44  1055.2   15.88  1217.8   15.34
  1232.9   18.57  1266.7   13.57 1593.11   13.23  1593.7   12.08  1631.7   12.08
 1632.71   13.71  1876.6   13.22  1908.1   14.88  1955.4    13.2    2046   17.67
  2061.7    16.7  2160.2   20.03  2550.9   22.75  2758.9   23.12  3194.6   20.81
#Mann= 3 ,0,0
       0     .15       0 1593.11     .05       0 1632.71     .15       0
Bank Sta=1593.11,1632.71
XS Rating Curve= 0 ,0
Exp/Cntr=0.3,0.1

Type RM Length L Ch R = 1 ,1492    ,900.9,900.9,900.9
BEGIN DESCRIPTION:
Maple Swamp 1.0
END DESCRIPTION:
XS GIS Cut Line= 4
      2608319.78       755291.44      2608616.23       754565.64
      2608372.92       753532.42      2606653.49       752490.46
#Sta/Elev= 30
       0   24.98    38.7   23.74   172.7   24.44     279   21.75   303.8    22.8
   405.6   20.33     435   17.74   448.4   19.18     539    16.9   795.8   18.25
   913.3   13.82  1075.6   14.72  1247.5   13.14 1825.03   12.52  1826.5   11.86
  1864.5   11.86 1864.95   12.77  2008.7   12.39  2055.5   14.09  2102.4   13.15
  2201.2   14.03  2247.3   12.51    2301   13.53  2374.6   12.37  2807.4   13.22
  3064.6   12.22  3217.8   13.51  3244.7   18.26  3539.4   22.03    3856   22.09
#Mann= 3 ,0,0
       0     .15       0 1825.03     .05       0 1864.95     .15       0
Bank Sta=1825.03,1864.95
XS Rating Curve= 0 ,0
Exp/Cntr=0.3,0.1

Type RM Length L Ch R = 1 ,591     ,0,0,0
BEGIN DESCRIPTION:
Maple Swamp 0.5
END DESCRIPTION:
XS GIS Cut Line= 4
      2609297.06       755253.57      2608755.97       752778.34
      2608272.43       752502.03      2606614.53       752317.82
#Sta/Elev= 30
       0   21.02      98   21.94   198.8   20.72     323    17.1     370   13.69
   400.3   13.22  1128.8   13.78    1213   12.53  1742.3   11.88    1804   13.53
  1978.7   11.68  2136.5   13.69  2203.7   11.94  2257.4   13.16  2324.6   11.74
    2402    13.6  2465.6   11.81 2781.76    12.4  2782.7    10.7  2820.7    10.7
 2821.36   12.09  3107.6   11.59  3294.5   12.99  3784.2   11.76  3952.5   13.75
  4153.9   13.16  4170.4   13.72  4196.8   17.42  4533.3   21.66  4758.7   21.75
#Mann= 3 ,0,0
       0     .15       0 2781.76     .05       0 2821.36     .15       0
Bank Sta=2781.76,2821.36
XS Rating Curve= 0 ,0
Exp/Cntr=0.3,0.1
LCMann Table=0

Chan Stop Cuts=-1
Use User Specified Reach Order=0
Composite Channel Slope=5

--- MapleSwamp.g01 (geometry) ---

Geom Title=Duplicate Effective
Program Version=6.60

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
River Reach=Maple Swamp     ,Reach-1
Reach XY= 30
      2599537.86       777539.22      2600191.34       777563.86
      2601509.94       777021.38       2603516.3       777838.93
      2604284.17         777797.      2604939.52       777305.48
      2605392.23       777788.37      2606375.26       777827.18
      2607147.02       777474.06      2607845.55       776592.54
      2607789.75       775192.58      2608234.95       774272.83
      2608298.55       773649.78      2608098.52       772654.84
      2607752.86       771946.89      2607911.72       771559.59
      2607753.19       770823.93      2608769.52       770113.49
      2609093.13       768070.89      2608369.51       766441.66
      2605027.77       763868.03      2605364.15       760822.12
      2604191.53       758997.42      2604095.39       758343.69
      2604358.17       757075.95      2604982.63       755432.16
      2605301.02       755144.99      2606487.15       754845.34
      2608232.84       753765.46      2608584.43       752057.63

Type RM Length L Ch R = 1 ,37981   ,588,588,588
BEGIN DESCRIPTION:
Maple Swamp 60.0
END DESCRIPTION:
XS GIS Cut Line= 3
      2601231.68        778734.1      2601135.59       777096.71
      2600759.99       776262.47
#Sta/Elev= 30
  3359.8   48.98  3573.4   47.29  3684.5   48.86  3744.6   48.36  3774.6   46.82
  3924.9   46.25  3999.7   44.54  4123.7   45.45  4345.6   41.16  4465.8   42.84
  4525.9   42.05  4708.9   42.25  4926.7   43.44  4976.7   42.83  4990.6   41.16
  4991.4   39.66  5008.6   39.66  5009.4   41.16    5013   42.46  5174.1   43.66
  5237.7   42.52  5270.6   43.28  5437.3   42.61  5622.6   44.45  5630.6   44.65
  5674.8    50.3  5698.3   54.98  5742.8   59.16  5829.9   62.58  5914.9   62.55
#Mann= 3 ,-1,0
  3359.8     .15       0  4990.6     .05       0  5009.4     .15       0
Bank Sta=4990.6,5009.4
XS Rating Curve= 0 ,0
Exp/Cntr=0.3,0.1

Type RM Length L Ch R = 1 ,37393   ,759,759,759
BEGIN DESCRIPTION:
Maple Swamp 59.0
END DESCRIPTION:
XS GIS Cut Line= 3
      2601514.02       778978.47      2601709.72       777048.27
      2601654.32       776063.13
#Sta/Elev= 30
  3059.9   54.02  3129.8   51.27    3179   47.91  3239.3   47.03  3390.1   48.75
  3431.8   47.69  3465.4   48.41  3540.8   47.51    3571   45.88  3782.1   44.99
    3963   45.62  4324.8   42.62  4415.3   40.65  4656.5   41.11  4686.7   42.87
    4747   43.66  4909.2   43.07  4990.6   40.65  4991.4   39.15  5008.6   39.15
  5009.4   40.65  5016.7   42.08  5131.7   43.14  5211.7   41.46  5578.5   41.23
  5619.2   42.59  5718.8    49.2  5858.1   54.74  5949.8    61.4  5986.7   62.85
#Mann= 3 ,-1,0
  3059.9     .15       0  4990.6     .05       0  5009.4     .15       0
Bank Sta=4990.6,5009.4
XS Rating Curve= 0 ,0
Exp/Cntr=0.5,0.3

Type RM Length L Ch R = 1 ,36634   ,129,129,129
BEGIN DESCRIPTION:
Maple Swamp (SCL RR) US
END DESCRIPTION:
XS GIS Cut Line= 3
      2603048.88       778939.54      2602400.43       777356.93
      2601843.97       776137.06
#Sta/Elev= 30
  3289.7   42.43  3357.5   43.09  3375.7   42.69  3426.5    43.8  3472.5   43.14
  3495.5   43.69  3518.5   43.15  3656.5   43.68  3679.4   42.82  3797.1   43.31
  4065.9    42.1  4092.5   41.27  4462.7    41.7  4704.9   39.12    4970   39.35
  4987.5    38.1    4993    35.1    5007    35.1  5012.5    38.1  5013.1   39.81
    5228    39.6  5352.8    40.7  5642.8      40  5909.9   40.89  6043.5   43.47
  6094.8   43.46  6177.1   45.35  6222.6   49.43  6281.8   50.83  6340.8   54.65
#Mann= 3 ,-1,0
  3289.7     .15       0  4987.5     .05       0  5012.5     .15       0
#XS Ineff= 2 , 0
       0    4950    40.1    5050       0    40.1
Permanent Ineff=
       F       F
Bank Sta=4987.5,5012.5
XS Rating Curve= 0 ,0
Exp/Cntr=0.5,0.3
